HEC-RAS study SNCHOCRK.prj: SNCHOCRK

--- SNCHOCRK.g01 (geometry) --- (continued)

Type RM Length L Ch R = 1 ,3474.1  ,311.3,337.2,362.8
XS GIS Cut Line= 4
     1567625.682       357905.72     1567726.377       357897.04
     1567899.988      357808.498     1567990.266      357794.609
#Sta/Elev= 27
       0  728.63     9.2  723.89    27.6  713.94    45.9  704.31    64.3  694.99
    82.7  685.99    91.9  681.73   101.1  678.02   110.8  674.92   120.6  672.91
   154.4666.8474   169.3  663.89     179  662.23   188.8  661.61   198.5   662.3
   208.3  664.58     218  667.42   227.7  669.68   237.5  671.44     257  674.37
     296  679.98   305.1  681.87   314.2     685   323.4  688.96   332.5  693.12
   359.9  705.33   387.3  717.84
#Mann= 3 , 0 , 0
       0      .1       0   154.4    .045       0     218      .1       0
Bank Sta=154.4,218
XS Rating Curve= 0 ,0
Exp/Cntr=0.3,0.1

Type RM Length L Ch R = 1 ,3136.9  ,556.5,577.3,597.5
XS GIS Cut Line= 3
     1567570.127      357949.123     1567901.724       358209.54
     1568032.084      358368.517
#Sta/Elev= 30
       0  746.08     9.8  744.55    19.6  742.12    39.2  735.32      49  732.08
    58.8  728.99   107.9  714.09   147.1  701.91   176.5  693.15   196.1  687.68
   205.9  685.13   215.7  682.83   225.5  680.89   313.8   666.5   326.7664.2842
   343.2  661.17     353  660.17   362.8  660.45   372.6  661.92   382.4  664.34
   392.2  667.44     402  672.78   411.8  679.95   421.6  687.51     451  709.33
   460.8   715.5   470.6  720.99   558.7  768.22   597.8   788.6   627.2  803.41
#Mann= 3 , 0 , 0
       0      .1       0   326.7    .045       0   392.2      .1       0
Bank Sta=326.7,392.2
XS Rating Curve= 0 ,0
Exp/Cntr=0.3,0.1

Type RM Length L Ch R = 1 ,2559.6  ,447.3,446.6,445.5
XS GIS Cut Line= 3
     1567398.252      358006.415     1567354.849       358209.54
     1567357.171      358674.506
#Sta/Elev= 30
       0  744.28     9.4  744.16    18.9  743.27    28.3   741.1    66.1  729.19
    94.4  719.77   132.2  706.47   188.8  686.03   198.3  682.81   207.7  680.23
   236.8  674.79   246.5  673.44   275.5  670.79   314.3  668.51     324  667.55
   333.6  665.46   343.3  662.04     353  659.86   362.7  659.42   372.4   659.4
   382.1   659.4   391.8   660.3   401.4  663.33   430.5  675.89   469.3  692.99
   517.7  714.47   546.8  727.66   585.5  745.88   643.6  774.95   672.7  788.94
#Mann= 3 , 0 , 0
       0      .1       0   343.3    .045       0   401.4      .1       0
Bank Sta=343.3,401.4
XS Rating Curve= 0 ,0
Exp/Cntr=0.3,0.1

Type RM Length L Ch R = 1 ,2113    ,478.6,473.2,467.5
XS GIS Cut Line= 4
     1566877.418      358173.081     1566913.877      358261.623
     1566922.557       358459.54     1566974.641       358584.54
#Sta/Elev= 30
       0  712.74    19.2  706.13    47.9  696.04    57.4   692.6   114.6  672.59
   124.1  669.22   133.5  665.49   142.9  661.73   152.4  659.64   161.8  659.83
   171.2  661.88   180.7  664.87   190.1  667.39   199.5  668.49     209  668.32
   218.4  667.99   227.8  668.03   237.3  668.46   246.7  669.12   256.1  670.24
   265.6  671.97   284.4  676.28   303.5  680.52   313.2   683.2   322.9  686.64
   351.9  697.69   380.9  708.43   409.9  719.34   419.6  722.79   429.3   725.9
#Mann= 3 , 0 , 0
       0      .1       0   133.5    .045       0   180.7      .1       0
Bank Sta=133.5,180.7
XS Rating Curve= 0 ,0
Exp/Cntr=0.3,0.1

Type RM Length L Ch R = 1 ,1639.8  ,150.3,149.8,149.3
XS GIS Cut Line= 4
     1566467.696      358259.887     1566436.446      358341.484
     1566495.474      358541.137     1566566.654      358653.984
#Sta/Elev= 29
       0   717.1     9.7  715.14    19.4   712.6    29.1  708.71    38.8  703.85
    58.2  694.35      68  689.63    77.7  684.98   106.3  671.66   115.8  666.99
   125.2  662.52   134.7  659.93   144.2  659.94   153.6  661.74   163.1  664.43
   172.5666.5574     182  668.14   191.5  669.25   200.9  670.16   210.4  670.96
   238.8   673.1   276.6  676.55   305.1  678.98   362.3   683.3   371.8  684.09
   381.3   685.2   390.9  687.06   400.4  689.98     429  699.73
#Mann= 3 , 0 , 0
       0      .1       0   115.8    .045       0   172.5     .08       0
Bank Sta=115.8,172.5
XS Rating Curve= 0 ,0
Exp/Cntr=0.3,0.1

Type RM Length L Ch R = 1 ,1490    ,317.7,312.7,306.7
XS GIS Cut Line= 4
     1566177.766      358306.762     1566281.932      358353.637
     1566365.266      358614.054     1566389.571      358759.887
#Sta/Elev= 30
       0  719.27      19  717.41    57.1  714.44    76.2  712.62    85.7  711.37
    95.2  709.14   104.7  703.04   114.2  693.55     124   680.8   133.8  671.19
   143.5  666.08   153.3   663.3     163  661.57   172.8  660.45   182.6  659.61
   192.4  659.14   202.1  659.84   211.9  662.62   221.6  666.72   231.4  669.71
   241.2  671.02   329.1  674.94   368.1  676.88   415.4  680.03   443.1  682.71
   452.3  684.23   461.6  686.73   480.1   692.8     517  705.65   535.5  711.67
#Mann= 3 , 0 , 0
       0      .1       0   143.5    .045       0   221.6     .08       0
Bank Sta=143.5,221.6
XS Rating Curve= 0 ,0
Exp/Cntr=0.3,0.1

Type RM Length L Ch R = 1 ,1177.3  ,314.3,320.6,326.3
XS GIS Cut Line= 4
     1565955.067      358414.541     1565988.266      358501.076
     1566088.715       358664.34     1566145.915      358833.043
#Sta/Elev= 30
       0   706.4    37.1  700.03    64.9  694.87    74.2  693.29    83.4  692.54
    92.7   692.1   102.3  689.89   111.8  684.46   121.4  677.13     131  670.21
   140.6  665.64   150.2   662.7   159.8  660.46   169.4  659.48     179  660.21
   188.5   662.6   198.1  665.75   207.7  668.42   217.3  670.34   226.9   671.6
     246  673.07   265.2  674.28   312.5  676.68   340.6  678.31   378.1  681.06
   387.5  682.22   396.9  684.36   406.3  687.66   453.1   706.7   462.5  709.74
#Mann= 3 , 0 , 0
       0     .08       0   140.6    .045       0   188.5     .07       0
Bank Sta=140.6,188.5
XS Rating Curve= 0 ,0
Exp/Cntr=0.3,0.1

Type RM Length L Ch R = 1 ,856.6   ,349.5,347.9,346.1
XS GIS Cut Line= 5
     1565790.613      358539.401      1565747.21       358678.29
     1565813.182      358900.512     1565912.141      359044.609
     1566136.678      359416.484
#Sta/Elev= 30
       0  685.05    19.4  681.38    29.1  681.06    77.6  683.26   116.4  681.85
   155.2  676.03   193.8  667.23   213.1  661.15   222.8   659.4   232.4   659.6
   260.4665.5733     300  668.87   377.3  680.36     387  682.24   416.2  691.58
   425.9  693.78   464.7  698.77   503.6  699.12   561.8  697.32   600.4  690.63
   658.3  677.99   696.9  676.55   774.2  678.12   851.4  681.82     861  683.61
   899.6  698.77   909.3   701.3   938.3  704.38   957.6  702.67   986.5  694.52
#Mann= 3 , 0 , 0
       0      .1       0   193.8    .045       0   260.4     .07       0
Bank Sta=193.8,260.4
XS Rating Curve= 0 ,0
Exp/Cntr=0.3,0.1

Type RM Length L Ch R = 1 ,508.7   ,392.5,389.9,387.3
XS GIS Cut Line= 3
     1565341.539      358645.651     1565400.566      358756.762
     1565709.594      359576.206
#Sta/Elev= 30
       0  728.73     9.7  726.69    19.4  723.73      29  719.64   125.8  674.47
   135.7  670.74   145.5  668.84   194.7  668.17     208666.6536   214.4  665.38
   234.1  659.86   243.9  658.88   253.7  659.95     278665.3936   293.1  667.65
   352.1  671.41   401.3  672.94   450.5  672.01   470.2  672.35   519.4     677
   657.2  676.88   696.6  677.75   735.9  679.54     854  680.58   873.7  680.16
   903.2   678.7     913  679.05   942.6  682.21   952.4  682.69  1001.6  683.43
#Mann= 3 , 0 , 0
       0      .1       0     208    .045       0     278     .07       0
Bank Sta=208,278
XS Rating Curve= 0 ,0
Exp/Cntr=0.3,0.1

Type RM Length L Ch R = 1 ,118.9   ,115.5,118.9,122.2
XS GIS Cut Line= 3
     1565081.122       358690.79     1565056.816      358954.679
     1565338.066      359499.817
#Sta/Elev= 30
       0  697.78    68.7  688.72     157  678.31   186.5  675.13   196.3  674.41
   206.1   674.1   215.9   673.3   225.8  671.67   235.6  669.71   255.2  664.98
   274.7  659.38   284.5  658.16   294.2     658     304  659.03   323.4  665.12
   325.2665.4781   333.2  667.07   352.6  668.49   401.3  672.66   420.8  673.92
   440.3  674.68   498.7   675.7   547.4  676.95   566.8  677.19   596.1  676.79
   625.3   676.8   683.7  676.22   703.2  676.31   742.1  677.42   878.4   680.6
#Mann= 3 , 0 , 0
       0      .1       0   255.2    .045       0   325.2      .1       0
Bank Sta=255.2,325.2
XS Rating Curve= 0 ,0
Exp/Cntr=0.3,0.1

Chan Stop Cuts=-1
Use User Specified Reach Order=0
Composite Channel Slope=5

--- SNCHOCRK.g02 (geometry) ---

Geom Title=USGS 10m DEM_copy
Program Version=4.10

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
River Reach=SNCHOCRK        ,Main

Type RM Length L Ch R = 1 ,52404.8 ,135.6,156.4,165.7
XS GIS Cut Line= 3
     1570080.522      327703.832      1570148.23      327628.311
     1570603.959      327432.999
#Sta/Elev= 30
       0  890.92    18.4   886.1    27.7  883.19    36.9  879.51    55.3  868.92
      83  850.66   101.4  839.07   111.2  834.17   120.9   830.4   130.6  828.09
   140.3  827.13   159.8  825.86   179.2  823.79   188.9  822.86   198.6  822.46
   218.1   822.7   247.3  823.34   295.9  822.73   334.8  825.48   373.6  826.33
   402.8  828.79   441.7  833.89   451.4  837.94   490.3  862.82   509.8  874.01
   519.5  878.95   529.2  883.17   538.9  886.66   568.1  896.39   597.2  902.22
#Mann= 3 , 0 , 0
       0     .07       0   179.2    .045       0   218.1     .06       0
Bank Sta=179.2,218.1
XS Rating Curve= 0 ,0
Exp/Cntr=0.3,0.1

Type RM Length L Ch R = 1 ,52248.4 ,157.1,191.2,187.7
XS GIS Cut Line= 2
     1570136.605      327750.107     1570607.525      327604.707
#Sta/Elev= 30
       0  885.39     9.7  882.17    19.3  877.77    38.7  866.96    96.6  833.63
   106.3   829.3     116  826.93   125.6  826.11     211 822.746   222.3   822.5
   231.9  822.78     242 823.436   280.2  827.23   289.9  828.03   299.6  828.47
   309.2   828.5   318.9  828.02   328.6  827.21   338.2  826.85   347.9  827.41
   357.6  828.63   376.9  831.96   386.6  832.98   405.9   833.8   415.5  834.59
   434.9  836.84   454.2  839.77   463.9  841.53   483.2     846   492.9  848.97
#Mann= 3 , 0 , 0
       0     .06       0     211    .045       0     242     .06       0
Bank Sta=211,242
XS Rating Curve= 0 ,0
Exp/Cntr=0.3,0.1

Type RM Length L Ch R = 1 ,52057.2 ,367.1,361.8,345.9
XS GIS Cut Line= 3
     1570197.709      327854.874     1570296.667      327810.603
     1570619.584      327709.041
#Sta/Elev= 30
       0  881.19       9  877.95    18.1  873.39    36.1  863.02    72.3  842.46
    81.3  837.14    90.3  832.09    99.4  828.43   108.4  826.55   118.1  825.73
   137.4  824.68   147.1  824.18   176.1  822.99   224.5  822.68   263.2  822.72
   291.5  822.88   311.5  822.29   321.2  822.12   330.9  823.89   340.5  828.07
   350.2  831.87   359.9   833.8   369.6  834.61   379.2  835.68   388.9  837.66
   398.6   841.2   408.2  846.14   417.9  851.45   427.6  856.47   446.9  865.92
#Mann= 3 , 0 , 0
       0     .06       0   291.5    .045       0   330.9     .06       0
Bank Sta=291.5,330.9
XS Rating Curve= 0 ,0
Exp/Cntr=0.3,0.1

Type RM Length L Ch R = 1 ,51695.4 ,456.6,482,458.6
XS GIS Cut Line= 2
     1570195.105      328018.936     1570635.209      327893.936
#Sta/Elev= 30
       0  889.22     9.7  887.46    29.2  885.31    38.9  883.36    48.7  880.58
    58.4  876.91    68.1  872.31    77.9   866.4    87.6  859.74   107.1   845.4
   116.8  838.52   126.6  832.35   136.3   826.6     146  821.57   155.8  818.68
   165.5  818.13   175.2  818.72     185  820.18   194.7  821.56   204.4  822.17
   253.1  824.25   282.3  825.14   360.2  826.17   369.9  827.62   389.4  833.63
   399.1   834.9   408.8  835.54     438  839.21   447.8  840.64   457.5  843.02
#Mann= 3 , 0 , 0
       0     .08       0     146    .045       0     185     .06       0
Bank Sta=146,185
XS Rating Curve= 0 ,0
Exp/Cntr=0.3,0.1

Type RM Length L Ch R = 1 ,51213.4 ,92.1,67.8,41.5
XS GIS Cut Line= 4
     1570239.376      328261.124     1570327.917      328334.041
      1570679.48      328219.457     1570781.042      328143.936
#Sta/Elev= 30
       0  880.55    19.1  872.99    57.4  854.32    76.5  842.72    95.6  830.36
   105.1  824.87   114.7   820.6   134.2   816.9     147  815.33   163.4   814.6
   192.6  814.77     212  815.71   241.2  816.12   309.3  819.43     358  824.17
   396.9  826.34   426.1  829.47   435.8  830.19   455.3  830.18     465  830.72
   474.7  832.21   484.5  834.44   494.2   839.6   523.4  859.72   533.1  864.73
   542.9  869.09   572.1  880.14   591.6  889.09   601.3  893.01     611  896.17
#Mann= 3 , 0 , 0
       0     .08       0     147    .045       0   192.6     .06       0
Bank Sta=147,192.6
XS Rating Curve= 0 ,0
Exp/Cntr=0.3,0.1

Type RM Length L Ch R = 1 ,51145.6 ,63.9,63.5,65.1
XS GIS Cut Line= 6
     1570210.187      328649.904      1570247.08      328539.227
     1570490.135      328289.661     1570516.177      328285.321
     1570693.043      328261.449     1570815.656      328343.915
#Sta/Elev= 30
       0  863.66      68  836.83    77.8   833.9    87.5  832.38   116.7  830.65
   155.4   829.1   213.4  825.78   252.1  821.58   271.5  821.23   290.8  819.96
   319.9  815.52   339.2  814.65   358.6  815.08   397.3  816.58     436   817.2
   491.4  819.65     529  822.73   585.4  826.06   594.8  827.42   613.5   832.1
   622.9  833.67   651.1  833.62   669.9  834.67   679.1  836.33   688.4  838.72
   706.8  844.37   725.3  849.19   771.5  864.69   799.2  875.61   817.7  882.13
#Mann= 3 , 0 , 0
       0     .08       0   319.9    .045       0   358.6     .06       0
Bank Sta=319.9,358.6
XS Rating Curve= 0 ,0
Exp/Cntr=0.3,0.1

Type RM Length L Ch R = 1 ,51082.1 ,169.6,294.3,322.8
XS GIS Cut Line= 6
     1570250.335      328698.732     1570287.227      328588.055
     1570530.283      328338.489     1570556.325      328334.149
     1570733.191      328310.278     1570855.804      328392.743
#Sta/Elev= 30
       0  876.15     9.7  871.39    29.2  860.72    38.9  856.31    87.5  839.06
   106.9  833.87   126.3  830.51   145.7  828.29   203.8  824.83   261.8  823.26
   290.8  821.56   310.2  819.23   329.6  815.26   339.2  814.15   358.6  815.39
   377.9   816.8     436  818.54     465  820.34     529  823.12   547.8  825.17
   585.4  832.09   604.2  833.21   622.9   835.2   632.3  837.28   660.5  848.82
   669.9  852.04   697.6  863.14   743.8  880.68   808.4  899.73   817.7  902.91
#Mann= 3 , 0 , 0
       0     .06       0   329.6    .045       0   358.6     .06       0
Bank Sta=329.6,358.6
XS Rating Curve= 0 ,0
Exp/Cntr=0.3,0.1

Type RM Length L Ch R = 1 ,50787.9 ,348.4,302.9,309.4
XS GIS Cut Line= 4
     1570259.341      328777.834     1570329.654      328652.834
     1570670.799      328548.667     1570832.258      328530.438
#Sta/Elev= 30
       0  885.03    19.1  882.27    28.7  879.99    38.2  876.77    57.4   869.2
   105.2  847.95   114.7  843.88   124.3  840.36   162.7  830.88   172.3  828.92
   191.6  826.46   239.8   821.9   336.2  814.45   384.4  812.13   403.7  812.82
     423  814.22   432.6  814.19     453 811.605   461.6  811.33     470 813.351
   471.2  813.64   490.5  823.62   500.1  827.01   519.2   831.3     567  850.76
   586.1   859.5   595.7  864.72   614.8   876.7   633.9  889.97   662.6  909.04
#Mann= 3 , 0 , 0
       0     .06       0     453    .045       0     470     .07       0
Bank Sta=453,470
XS Rating Curve= 0 ,0
Exp/Cntr=0.3,0.1

Type RM Length L Ch R = 1 ,50484.9 ,316.4,349.2,378.3
XS GIS Cut Line= 3
      1570398.99      328839.791     1570690.873      328845.217
     1570746.212       328818.09
#Sta/Elev= 30
       0  834.01     9.7  829.48    19.5  825.13    29.2  821.94    38.9  820.43
    48.7  819.64    58.4  818.96    68.1  818.32    77.8  817.83     146  816.18
   155.7  815.85   165.4  815.38   175.2  814.73   194.6  813.18   204.4  812.52
     231 810.936   233.6  810.79   243.3  810.82     252 811.421   262.7  812.28
   272.5  813.24   282.2  814.82   291.9     817   300.7  818.79   309.5  820.02
   318.4  821.65   327.2  824.85     336  828.81   344.8  833.07   353.6  837.44
#Mann= 3 , 0 , 0
       0     .06       0     231    .045       0     252     .07       0
Bank Sta=231,252
XS Rating Curve= 0 ,0
Exp/Cntr=0.3,0.1

Type RM Length L Ch R = 1 ,50135.7 ,463.5,470.6,422.6
XS GIS Cut Line= 3
     1570476.029      328977.595     1570682.193      329179.418
     1570817.826      329195.694
#Sta/Elev= 29
       0  818.39     9.6  818.05    38.5   816.6    57.7  815.73   115.4  813.32
     125  812.81   144.2  811.52   182.6  809.25     202  807.97     207 807.777
   211.6   807.6   221.2  807.69     227 808.119   230.8   808.4     250  810.37
   259.7  810.87   269.3  811.18   278.9  811.61   288.5  812.41   298.3   813.5
     308  814.35   327.5  815.59   337.3  816.35   356.8  818.31   366.6  819.12
   376.3  819.39   395.8  819.39   405.6   819.3   425.1  818.97
#Mann= 3 , 0 , 0
       0     .06       0     207    .045       0     227     .06       0
Bank Sta=207,227
XS Rating Curve= 0 ,0
Exp/Cntr=0.3,0.1

Type RM Length L Ch R = 1 ,49665.1 ,335.1,330.2,350.1
XS GIS Cut Line= 4
     1570357.757      329414.878     1570408.755      329444.175
     1570496.646      329446.345      1570559.58      329399.687
#Sta/Elev= 28
       0  832.14     9.8  828.23    19.6   824.3    29.4  820.41    34.9  818.01
    39.2  816.14      49  810.82    58.8  805.73      61 805.119    68.6  803.01
    78.4  802.58      84 802.921    88.1  803.17    97.9  804.03   104.9  804.67
   107.7  804.92   117.4  805.77   127.2   806.6     137  807.42   146.7  808.16
   156.5  808.76   166.3  809.39   176.1  810.05   185.9  810.69   195.7  811.21
   205.5  811.68   215.3  812.05   225.1  812.31
#Mann= 3 , 0 , 0
       0      .1       0      61    .045       0      84     .08       0
Bank Sta=61,84
XS Rating Curve= 0 ,0
Exp/Cntr=0.3,0.1

Type RM Length L Ch R = 1 ,49334.9 ,146.5,113.7,77.5
XS GIS Cut Line= 5
     1570287.227      329788.142     1570342.566      329719.783
     1570393.564      329733.889     1570504.241      329784.887
     1570702.809      329787.057
#Sta/Elev= 29
       0  864.87     9.8  859.69    19.5  853.06    29.3     846    48.9  831.32
    58.6  824.28    68.4  817.74    78.2  813.71      88  811.92    96.8  810.86
   114.4  809.03   150.2  805.68   159.6  804.45     171   802.3   178.4  801.04
   187.7  801.24     205 803.659   206.5  803.86   215.9  804.73   225.2  805.27
     244  806.11   262.7  806.76     310  807.96   328.9  808.59   338.4  809.05
   357.3  810.09   432.9  813.98   451.8  815.16   461.3  816.15
#Mann= 3 , 0 , 0
       0      .1       0     171    .045       0     205     .07       0
Bank Sta=171,205
XS Rating Curve= 0 ,0
Exp/Cntr=0.3,0.1

Type RM Length L Ch R = 1 ,49221.3 ,289,293,279.2
XS GIS Cut Line= 4
      1570324.12      329873.863     1570385.969      329849.991
     1570494.476      329816.354     1570683.278      329797.908
#Sta/Elev= 23
       0     867     9.5  862.32    18.9  854.69    28.4  846.52    37.9   837.9
    47.4  828.96    56.8  819.21    66.3  809.17      73 804.346    75.8  802.33
    85.2  800.92      88 801.274    94.7  802.12   104.2  803.09   113.6  803.73
     142  805.02     161  805.76   179.9  806.38   189.4  806.59   227.3  807.14
   246.3  807.61   265.3  808.56   369.6  814.57
#Mann= 3 , 0 , 0
       0     .06       0      73    .045       0      88     .06       0
Bank Sta=73,88
XS Rating Curve= 0 ,0
Exp/Cntr=0.3,0.1

Type RM Length L Ch R = 1 ,48928.3 ,174.5,214.7,266.2
XS GIS Cut Line= 4
     1570325.407      330067.815     1570515.294      330110.133
     1570609.696      330056.964     1570725.798      330053.709
#Sta/Elev= 30
       0  856.03     9.7  849.57    19.4  842.14    38.9  826.29    48.6  819.06
    58.4  812.73    68.1  808.23    77.8  806.35    97.3  805.45   116.7  805.01
   165.4  804.63   194.6   804.1   203.6  803.59   212.6  802.56     220  801.36
   221.6   801.1   230.7  800.43   239.7  801.15     247 802.107   257.8  803.25
   322.2   807.1   331.9  807.57   351.3  808.11     361   808.5   370.6  809.15
   380.3  810.14     390  811.66   399.7  814.02   409.4  817.12     419  819.02
#Mann= 3 , 0 , 0
       0     .06       0     220    .045       0     247     .06       0
Bank Sta=220,247
XS Rating Curve= 0 ,0
Exp/Cntr=0.3,0.1

Type RM Length L Ch R = 1 ,48713.6 ,281.2,274.7,269.3
XS GIS Cut Line= 3
     1570304.588      330158.151     1570519.432      330238.446
     1570661.576      330319.826
#Sta/Elev= 30
       0  847.37     9.6  841.12    19.1  834.73    38.2  822.04    47.8   815.9
    57.3  810.87    66.9  808.11    76.4  807.17    95.6  806.73   124.2  806.58
   162.5  806.85   191.1  806.88   200.7  806.78   219.8  806.34     239   805.5
   258.3   804.4   267.9  803.71   277.5  802.85   287.2  801.79   296.8  800.56
   306.4  799.22     308 799.068   316.1   798.3   325.7  798.51   335.3  801.22
     345  806.29   354.6  811.95   364.2  816.08   383.5  818.56   393.2  822.47
#Mann= 3 , 0 , 0
       0     .07       0     308    .045       0   335.3     .06       0
Bank Sta=308,335.3
XS Rating Curve= 0 ,0
Exp/Cntr=0.3,0.1

Type RM Length L Ch R = 1 ,48438.9 ,341.9,336.4,347.6
XS GIS Cut Line= 4
     1570209.102      330421.823     1570455.413      330520.564
     1570518.347      330547.691      1570555.24      330571.562
#Sta/Elev= 30
       0  818.86     9.8  816.99    19.7  815.44    39.3  812.52    49.1  810.88
      59  809.65    68.8  808.96    78.6  808.42    98.3  807.75   108.1  807.59
   127.8  807.65   167.1  808.17   186.7  808.16   196.6  807.97   206.4  807.65
   216.2  807.13   235.9  805.63   245.7  804.65   255.5  803.37   265.4  801.02
     275  798.13     285  796.45   294.7  796.62     300 797.123   314.3  798.63
   324.1  799.87   333.9  802.88   342.7  806.96     369  819.82   377.8  822.46
#Mann= 3 , 0 , 0
       0     .06       0     275    .045       0     300     .06       0
Bank Sta=275,300
XS Rating Curve= 0 ,0
Exp/Cntr=0.3,0.1

Type RM Length L Ch R = 1 ,48102.4 ,433.5,418.5,383.6
XS GIS Cut Line= 4
     1570184.146      330754.939     1570248.165      330754.939
     1570404.415      330863.446     1570485.795      330927.465
#Sta/Elev= 30
       0  835.75     9.2  829.68    18.3  823.42    27.4  816.87    36.6  810.54
    45.7  805.59    54.9  802.25      64  799.64    73.5  797.13      82 795.162
      83  794.93    92.6  794.16     100 794.534   102.1  794.64   111.6   795.6
   121.1  796.73   130.6  797.64   140.1  798.14   159.1  798.46   206.7  798.56
   216.2  798.68   225.7  798.94   254.2  800.15   263.7  800.71   273.1  801.58
   282.5  803.54   291.9   806.1     339   820.4   348.4  823.14   357.8   825.4
#Mann= 3 , 0 , 0
       0     .07       0      82    .045       0     100     .06       0
Bank Sta=82,100
XS Rating Curve= 0 ,0
Exp/Cntr=0.3,0.1

Type RM Length L Ch R = 1 ,47683.9 ,182.5,221.3,246.1
XS GIS Cut Line= 2
      1570101.68       331168.35     1570389.224      331165.095
#Sta/Elev= 23
       0  842.82     9.6  836.98    28.8  825.02    38.3  818.99    47.9  812.78
    67.1  798.78      74 795.697    76.7  794.49    86.3  793.63      91  794.08
    95.8  794.54   105.4  795.98     115  797.14   124.6   797.7   134.2  797.79
   153.4  797.56     163  797.54   172.5  797.73   191.7  798.49   210.9   799.4
   268.4   802.4     278  803.32   287.6  805.41
#Mann= 3 , 0 , 0
       0      .1       0      74    .045       0      91     .06       0
Bank Sta=74,91
XS Rating Curve= 0 ,0
Exp/Cntr=0.3,0.1

Type RM Length L Ch R = 1 ,47462.6 ,116.7,107.8,110.1
XS GIS Cut Line= 4
     1570110.361      331302.899     1570183.061      331363.663
     1570279.632      331410.321     1570400.075      331416.831
#Sta/Elev= 29
       0  834.56     9.5  830.68      19  826.67    28.4  823.21    37.9  820.22
    47.4  817.34    56.8  814.18    66.3  809.74    75.8  804.94    85.3  800.76
    94.8  797.35   104.5  795.28   114.2  793.59     124  792.47     133   791.8
   133.8  791.74   143.5  791.72   153.2  792.22     160 792.775   172.8  793.84
     202   796.1   220.6  797.71   229.8  798.71   239.1  799.86   276.2  804.72
   285.5  806.31   294.8  808.46   313.3  813.45   322.6  815.61
#Mann= 3 , 0 , 0
       0     .06       0     133    .045       0     160     .06       0
Bank Sta=133,160
XS Rating Curve= 0 ,0
Exp/Cntr=0.3,0.1

Type RM Length L Ch R = 1 ,47354.8 ,194.5,238,280.1
XS GIS Cut Line= 4
     1570114.701      331419.001     1570160.274      331464.574
      1570253.59      331518.828     1570510.954      331597.763
#Sta/Elev= 30
       0  809.38     9.2  804.24    18.4  800.11    27.6  797.73    36.8  797.14
    55.2  796.62    64.4  796.02    74.3  795.13    93.9  792.65     100  792.04
   103.7  791.67   113.5  791.62     122 792.245   152.8  794.75   191.6  797.39
   220.5  800.08   230.1  801.11   258.9  804.64   278.2  806.41   287.8  807.57
     307  811.18   316.6  811.99   326.2  813.12   335.8  815.27   345.4  817.71
   355.1  820.55   374.3  826.65   403.1  834.64   412.8  837.62   441.6   847.4
#Mann= 3 , 0 , 0
       0     .06       0     100    .045       0     122     .06       0
Bank Sta=100,122
XS Rating Curve= 0 ,0
Exp/Cntr=0.3,0.1

Type RM Length L Ch R = 1 ,47116.8 ,110.8,92.4,77.3
XS GIS Cut Line= 4
     1570048.512      331534.019     1570098.425      331640.356
     1570114.701      331738.012     1570251.623      331949.326
#Sta/Elev= 30
       0  797.18     9.8  795.63    19.6  795.25    68.5  795.18    88.1  794.83
   117.5  794.02   126.5  793.44   135.5  792.64     154   790.4   162.5  789.72
   171.5  789.56     181  789.84   189.5  790.69   207.5  793.14   216.5  794.06
   264.9  797.46   274.6  797.94   284.3  798.03   313.3   797.9     323  798.21
   332.7  799.66   342.4  802.43     352  805.94   361.7  808.21   381.1  808.64
   400.5  809.64   419.8  810.34   448.9  810.22   458.6  810.75   468.3  811.69
#Mann= 3 , 0 , 0
       0     .06       0     154    .045       0     181     .06       0
Bank Sta=154,181
XS Rating Curve= 0 ,0
Exp/Cntr=0.3,0.1

Type RM Length L Ch R = 1 ,47024.4 ,217.5,269.4,270.5
XS GIS Cut Line= 4
     1569935.867       331545.68     1569960.824       331627.06
     1570095.373      331835.393     1570097.543      331898.327
#Sta/Elev= 30
       0  837.97     9.5  833.56    18.9  828.98    28.4  824.24    37.8  819.29
    47.3     814    66.2  802.58    75.7  797.51    85.1  794.43    94.7  793.21
   104.2  792.98   132.8  792.82   151.9  792.28     171  791.32   199.6  789.31
     207 788.889   209.1  788.77   218.7  788.75   228.2   789.2     236 789.955
   256.8  792.18   285.4  794.92   304.5   796.4   333.1   798.3   351.1  799.18
   360.1  800.02   369.1  801.75   378.1  804.53   387.1  807.79   396.1  810.82
#Mann= 3 , 0 , 0
       0     .07       0     207    .045       0     236     .06       0
Bank Sta=207,236
XS Rating Curve= 0 ,0
Exp/Cntr=0.3,0.1

Type RM Length L Ch R = 1 ,46755   ,292.7,279.6,262.9
XS GIS Cut Line= 3
     1569795.893      331615.124      1569938.92      331880.156
     1569971.472      331966.962
#Sta/Elev= 30
       0  821.14     9.7  821.34    38.9  821.01    48.6  821.02    58.3  819.66
      68  816.38    77.7  810.76   106.9     791     112 788.808   116.6  786.83
   126.3  785.77     136   786.7     143 788.244   155.4  791.26   165.2  793.09
   174.9  794.15   184.6  794.72   194.3  795.13   213.7  795.41   233.2  794.95
   262.3  792.78     272   792.4   281.7   792.5   291.4  793.15   301.2  794.09
     329  797.19   338.2  798.41   347.5  800.22   356.8  802.72   393.9   814.3
#Mann= 3 , 0 , 0
       0      .1       0     112    .045       0     143     .06       0
Bank Sta=112,143
XS Rating Curve= 0 ,0
Exp/Cntr=0.3,0.1

Type RM Length L Ch R = 1 ,46475.4 ,187.9,214.5,238.5
XS GIS Cut Line= 4
     1569570.199      331729.056     1569615.808      331881.115
     1569733.842      331989.748      1569857.54      332061.363
#Sta/Elev= 30
       0  879.72     9.3   874.9    37.4  860.76    46.7  855.92      56  850.62
    74.7  839.35      84  834.26    93.4   829.5   102.7  824.91   112.1  820.42
   121.4  816.02   130.7  811.78   149.4  803.81   158.8  800.07   168.2  795.66
   177.6  790.77   187.1  786.13   196.5  783.48   205.9  783.36   215.4   784.3
   234.2   786.9   243.7  788.01   253.1  788.97     272  790.66   309.7  793.43
   404.9  799.61   433.5  801.83     443  802.71   452.6  804.06   462.1  806.51
#Mann= 3 , 0 , 0
       0      .1       0   187.1    .045       0   215.4     .08       0
Bank Sta=187.1,215.4
XS Rating Curve= 0 ,0
Exp/Cntr=0.3,0.1

Type RM Length L Ch R = 1 ,46260.9 ,189.4,162.7,142.3
XS GIS Cut Line= 4
     1569502.722      331984.323     1569520.083      332040.746
     1569562.401      332148.168     1569591.698      332261.015
#Sta/Elev= 21
       0  800.92     9.8  796.42    19.7  793.64    29.5  792.13    68.7   787.9
     105 783.641   107.1   783.4   116.8  782.92   126.4  783.13     132 783.696
     136   784.1   155.2  786.93   174.5  789.48   184.2  790.68   193.9  791.71
   203.6  792.56   223.1  793.89   242.5  794.82   252.2  795.12   271.6  795.36
   291.1  795.23
#Mann= 3 , 0 , 0
       0     .06       0     105    .045       0     132     .06       0
Bank Sta=105,132
XS Rating Curve= 0 ,0
Exp/Cntr=0.3,0.1

Type RM Length L Ch R = 1 ,46098.3 ,183.6,169.8,154.8
XS GIS Cut Line= 4
     1569332.865      331838.525     1569331.281      332109.106
     1569495.127      332281.632     1569571.082      332269.696
#Sta/Elev= 30
       0  915.48    19.3  903.68    67.6  875.29    77.3  870.13      87  865.56
    96.6  861.28   125.6  848.87   154.6   837.1   202.9  816.64   231.9  804.61
   241.6   800.7   251.3  796.99   260.9  793.69   270.6   791.2   280.1  789.82
   289.6  788.88   299.1  788.17   318.2  787.08   356.2  785.98   385.5  784.38
     400 783.426   413.3  782.72   422.9  782.66     433 783.293   460.9  786.02
   508.5  789.89   527.7  791.68   537.4  792.44   556.6  793.57   585.4  794.69
#Mann= 3 , 0 , 0
       0     .06       0     400    .045       0     433     .06       0
Bank Sta=400,433
XS Rating Curve= 0 ,0
Exp/Cntr=0.3,0.1

Type RM Length L Ch R = 1 ,45928.5 ,221.8,218.6,215.3
XS GIS Cut Line= 4
     1568955.261      332304.671     1569240.135      332297.908
     1569451.724      332419.435     1569568.911      332465.008
#Sta/Elev= 30
       0  908.24     9.8     906    29.5  900.81      59  892.34    68.8  889.26
   108.1  875.71   137.6  864.81   147.4  861.02   157.2  856.37     167  851.36
   186.7  841.88   196.5  836.77   206.4  831.18   216.2   824.8     226  817.58
   245.6  802.17   255.5   795.2   265.3  790.22   275.1   788.3   314.2  787.87
   333.8  787.32     363  785.84     393 783.725   411.8   782.5   421.6  782.53
     433 783.217   457.2  785.08   538.6  790.38   625.7  794.55   654.7  795.59
#Mann= 3 , 0 , 0
       0     .06       0     393    .045       0     433     .06       0
Bank Sta=393,433
XS Rating Curve= 0 ,0
Exp/Cntr=0.3,0.1

Type RM Length L Ch R = 1 ,45709.9 ,297.8,296.1,294.2
XS GIS Cut Line= 2
     1569092.566      332468.264     1569462.575      332652.725
#Sta/Elev= 22
       0  817.54    19.2  802.79    28.8  795.62    38.5     790    48.1  787.01
    57.7  786.06   105.8  783.51   134.6  781.75     143 781.383   153.8  781.29
     162 781.555   182.9  782.55   230.8  785.23   317.3  790.25   336.5  791.17
   346.1  791.32   355.8  791.27   365.4  791.12     375   790.8   394.2  789.61
   403.8  789.16   413.4  788.87
#Mann= 3 , 0 , 0
       0     .06       0     143    .045       0     162     .06       0
Bank Sta=143,162
XS Rating Curve= 0 ,0
Exp/Cntr=0.3,0.1

Type RM Length L Ch R = 1 ,45413.8 ,243.9,250.2,256.4
XS GIS Cut Line= 4
     1568930.891      332739.531      1568997.08      332746.041
     1569125.321       332804.36     1569393.333      332772.893
#Sta/Elev= 27
       0  828.41     9.5  824.69    47.5  809.03    85.3  793.83    94.7  789.55
   104.1  784.59     112 781.808   113.5  781.28   122.9  780.67   132.2  781.17
     142 782.183     151  783.16   160.4     784   169.8  784.55   188.6  785.42
     198  785.75     217  786.18   236.3  786.41   274.8  786.51   284.5   786.6
   303.8  786.91     323  787.36     352  788.28   380.9  789.48   409.8  790.92
     429  791.73   477.2  794.34
#Mann= 3 , 0 , 0
       0     .08       0     112    .045       0     142     .07       0
Bank Sta=112,142
XS Rating Curve= 0 ,0
Exp/Cntr=0.3,0.1

Type RM Length L Ch R = 1 ,45163.6 ,336.6,332.4,319.2
XS GIS Cut Line= 3
      1568836.49      332932.673      1569084.97      333085.668
     1569254.241      333084.583
#Sta/Elev= 28
       0  824.55     9.7  819.32    19.4  813.09    38.9  799.49    48.6  793.01
    58.4  786.67    68.1   781.6      75 780.192    77.8  779.62    87.5  779.26
    97.3  779.42     107  780.14     113 780.808   116.7  781.22   126.4  782.09
   145.9  782.96   155.6  783.27   165.4  783.48   184.8  783.55   223.7  783.13
   243.2  783.09   252.9  783.22   310.6   784.5   357.6   785.9   385.8  787.15
   395.2  787.71   414.1  789.09   461.1  792.81
#Mann= 3 , 0 , 0
       0     .08       0      75    .045       0     113     .06       0
Bank Sta=75,113
XS Rating Curve= 0 ,0
Exp/Cntr=0.3,0.1

Type RM Length L Ch R = 1 ,44831.2 ,212.3,173.7,143.6
XS GIS Cut Line= 5
     1568732.323      333256.024     1568774.641      333282.066
     1568857.106      333307.022     1569118.608      333303.767
     1569191.307      333326.554
#Sta/Elev= 29
       0  810.09    24.8  796.12    33.1  791.19    49.7  780.59      57 777.891
    59.3  777.04    68.8  776.44    78.4  777.02      80 777.183   107.1  780.03
   116.7  780.88   126.3  781.55   145.5   782.7   155.2   783.2   164.9  783.54
     194  784.15   213.3  784.16   281.1  782.72   290.8  782.63   300.5  782.64
   319.9  782.85   348.9  783.73   358.6  784.11   368.3  784.52   387.7  785.58
   406.9  786.92   416.4  787.66     464  791.74   473.6  792.95
#Mann= 3 , 0 , 0
       0     .08       0      57    .045       0      80     .06       0
Bank Sta=57,80
XS Rating Curve= 0 ,0
Exp/Cntr=0.3,0.1

Type RM Length L Ch R = 1 ,44657.5 ,238,311,380
XS GIS Cut Line= 4
     1568659.406      333453.073     1568741.003      333473.906
     1569079.545      333368.003     1569770.365      333460.921
#Sta/Elev= 30
       0  812.26    18.7  803.32    37.4   795.4    65.5  785.98    84.2  781.56
   122.6  776.49   141.7  775.78   160.9  777.02   208.8  781.22   247.2  783.49
   371.8  782.33   438.9  784.12   517.5     791   566.6  798.51   586.2   800.3
     596  801.86   605.8  804.46   694.2  832.41   733.5  849.27   743.3  852.25
   772.7  856.14   861.1  860.11   910.2  866.88   939.6  875.96   988.7  888.49
  1077.1  908.21  1086.9   908.5  1096.7  909.82  1126.2  917.16    1136   921.3
#Mann= 3 , 0 , 0
       0     .08       0   122.6    .045       0   160.9     .06       0
Bank Sta=122.6,160.9
XS Rating Curve= 0 ,0
Exp/Cntr=0.3,0.1

Type RM Length L Ch R = 1 ,44346.5 ,447.7,441.8,435.6
XS GIS Cut Line= 5
     1568640.309      333496.475     1568669.823      333524.253
     1568812.184      333769.045     1568906.614      333939.628
      1569285.99      334312.484
#Sta/Elev= 30
       0  808.15    24.3  796.63    40.5  790.01    69.8  780.66    79.6   778.8
   108.9  777.87   196.8  778.78   235.8  777.51     264 775.357   274.9   774.8
     287 775.953   304.2  778.12   401.7  786.51   479.7   795.3   528.4  810.79
   547.7   818.8   557.4  823.62   576.7  834.88   586.4  839.52     596  842.98
   625.1  851.26   654.1  858.79   683.1  864.73   731.4  871.15   808.8  884.35
   857.2  889.96   895.9  891.91   944.2  893.14  1011.9  891.95  1050.6     887
#Mann= 3 , 0 , 0
       0     .06       0     264    .045       0     287     .06       0
Bank Sta=264,287
XS Rating Curve= 0 ,0
Exp/Cntr=0.3,0.1

Type RM Length L Ch R = 1 ,43904.7 ,236.4,226.8,217
XS GIS Cut Line= 3
     1568315.859      333790.688     1568497.065       334054.36
     1568528.532       334210.61
#Sta/Elev= 30
       0   803.7     9.7  798.73    19.4  793.96    29.1  789.41    38.8  785.13
    48.5  781.22    58.2  778.06    67.9  776.06    87.3  773.44      99 772.019
   106.6  771.18   116.3  770.49     126   771.3     135 772.376   145.4  773.54
   155.1  774.27   184.2  775.98   203.6   776.9     223  777.51   252.1  777.74
   281.2  778.36   310.2  779.27   329.3   780.3   338.7  781.03   366.8  784.19
   404.3  788.15   432.4  791.39   441.8  792.29   460.6  793.54   479.3   794.3
#Mann= 3 , 0 , 0
       0     .08       0      99    .045       0     135     .06       0
Bank Sta=99,135
XS Rating Curve= 0 ,0
Exp/Cntr=0.3,0.1

Type RM Length L Ch R = 1 ,43677.8 ,312.4,348,367.4
XS GIS Cut Line= 3
     1568136.837      333947.864     1568324.337      334116.267
     1568475.378       334230.85
#Sta/Elev= 30
       0  800.71    19.4  794.21    29.1  791.06    38.8  787.58    48.5  782.05
    58.2  775.34      65 771.983    67.8   770.6    77.6  770.01      89  771.54
    96.9  772.68   106.6  773.83   135.7  776.82   145.4  777.67   155.1  778.38
   164.8  778.94   184.2  779.83   203.6  780.45   213.2  780.62   222.9  780.67
   232.6  780.59   242.3  780.39   280.5   779.2   289.9  779.09   299.4  779.23
   308.9  779.65   318.4  780.33   327.9  781.18   422.6  790.65   441.6   792.4
#Mann= 3 , 0 , 0
       0     .08       0      65    .045       0      89     .06       0
Bank Sta=65,89
XS Rating Curve= 0 ,0
Exp/Cntr=0.3,0.1

Type RM Length L Ch R = 1 ,43329.8 ,113.3,78.2,59
XS GIS Cut Line= 6
     1567158.386      333523.421     1567665.278      334062.842
     1567904.198        334137.1     1567904.198      334187.448
     1567951.073      334282.934     1568155.934      334505.156
#Sta/Elev= 30
       0  802.94     9.7  801.31    19.5  801.81    48.7  811.28    68.2  815.23
   136.4  819.56   253.2  821.06   409.1  816.67   506.5  823.55   545.4  821.11
   594.1  814.16   623.3  813.38   652.6  808.35   691.5  807.54   740.2  802.95
   769.1  806.78     798  807.46   884.6   803.1   990.4  792.75  1032.4  779.92
    1052 770.555  1060.1  768.35  1069.8  768.28    1082 769.504  1147.1   776.2
  1293.4  780.23  1361.6  784.72  1410.4  791.13  1420.1  793.99  1449.4  805.72
#Mann= 3 , 0 , 0
       0     .08       0    1052    .045       0    1082     .07       0
Bank Sta=1052,1082
XS Rating Curve= 0 ,0
Exp/Cntr=0.3,0.1

Type RM Length L Ch R = 1 ,43251.7 ,148.7,148.7,148.7
XS GIS Cut Line= 6
     1566759.949      333734.359     1567653.691      334184.748
      1567751.42      334203.073     1567810.448      334218.698
      1567961.49       334355.85     1568131.628      334609.323
#Sta/Elev= 30
       0  903.05    58.9  877.55   107.9  852.24   117.7  846.47   137.4  832.59
   147.2   828.5     157  829.03   186.4  836.95   215.9  840.98   255.1   848.7
   264.9   848.6   431.7  812.86   480.8  804.77   529.8  798.68   667.2  789.03
   902.7  783.37    1037  775.09  1135.1   774.8    1210 768.814  1219.6  768.26
    1240 770.123  1268.2  774.72    1307  777.09  1432.1  779.73  1498.9  779.02
  1527.5  780.62  1556.1  786.72  1584.8  791.19    1642  809.89  1670.6  820.54
#Mann= 3 , 0 , 0
       0     .08       0    1210    .045       0    1240     .06       0
Bank Sta=1210,1240
XS Rating Curve= 0 ,0
Exp/Cntr=0.3,0.1

Type RM Length L Ch R = 1 ,43103   ,170.2,141.9,127.1
XS GIS Cut Line= 5
     1567520.517      334274.253     1567631.628      334295.087
     1567690.656      334310.712     1567841.698      334447.864
     1568011.837      334701.337
#Sta/Elev= 30
       0  790.17     9.4  787.95    18.8  786.29    28.3  785.16    47.1  783.63
    65.9  782.94    94.2  780.67     113  779.77   147.9  778.79   174.1  779.19
   183.8  778.88   232.4  773.38   242.1  771.74     253 769.361   261.6  767.72
   271.3  767.72     286 770.181   290.7  770.98   310.1  772.46   378.1  774.79
   435.4  776.05   483.1  777.99   530.8  778.42   540.3  779.27   568.9   783.2
   616.6  788.42   635.7  789.81   645.2  791.29   654.8  794.28   683.4  805.07
#Mann= 3 , 0 , 0
       0     .08       0     253    .045       0     286     .06       0
Bank Sta=253,286
XS Rating Curve= 0 ,0
Exp/Cntr=0.3,0.1

Type RM Length L Ch R = 1 ,42961.1 ,182.1,198.7,194.5
XS GIS Cut Line= 4
     1567550.031       334472.17     1567636.837      334465.225
     1567853.851      334569.392     1567980.587      334677.031
#Sta/Elev= 30
       0  815.58     9.7  811.91    19.4  807.34      29   802.2    48.4  791.37
    58.1  786.24    67.7  781.56    77.4  777.25    87.1  773.51    96.7  770.07
     101 768.722   106.3  767.06     116   765.9   125.6  765.81   135.2  765.92
     140 766.148   144.9  766.38   212.3  771.08   250.8  773.58     270  774.73
   308.5  775.72   327.8  776.42   357.2  777.74   386.5  779.53     406  781.04
   425.6  782.74   435.4  783.72     455  785.88   474.5  788.28   494.1  790.19
#Mann= 3 , 0 , 0
       0     .08       0     101    .045       0     140     .07       0
Bank Sta=101,140
XS Rating Curve= 0 ,0
Exp/Cntr=0.3,0.1

Type RM Length L Ch R = 1 ,42762.4 ,138.6,145.7,153.8
XS GIS Cut Line= 5
     1567515.309      334616.267     1567569.128      334650.989
     1567770.517      334727.378     1567834.753      334774.253
     1567878.156      334850.642
#Sta/Elev= 30
       0  810.98    18.3  798.11    27.4  792.54    36.6  787.95    45.8  783.71
    54.9   779.1      64  773.31      74  767.27    83.6  765.81    93.4  765.88
      99 766.366   103.2  766.73     113  769.17   122.8  770.98   132.6  772.38
   142.4  773.23     162  774.23   181.5  774.76   201.1  774.69   259.9  772.84
   269.6  773.01   288.3  774.45   297.1  774.91   341.3  775.04   350.1  775.81
     359  776.91   378.5  780.67     398  783.43   427.3  786.97   446.8  788.74
#Mann= 3 , 0 , 0
       0     .08       0      74    .045       0      99     .08       0
Bank Sta=74,99
XS Rating Curve= 0 ,0
Exp/Cntr=0.3,0.1

Type RM Length L Ch R = 1 ,42616.7 ,350.2,356.3,364.5
XS GIS Cut Line= 4
     1567484.059      334749.948     1567515.309      334781.198
     1567605.587      334833.281     1567683.712        335074.6
#Sta/Elev= 23
       0  793.03     8.8  788.84    17.7  785.22    26.5  782.04    35.4  778.94
    44.2  775.72    53.7  771.34      62 767.879    63.1  767.42    72.6  765.46
    82.1  765.55      93 766.924     101   768.2   110.5   769.5     120  770.53
   129.5  771.34   138.9  771.95   167.9   773.4     207  774.89   304.5  777.82
   343.5  779.26   392.3  781.19   402.1   781.5
#Mann= 3 , 0 , 0
       0     .09       0      62    .045       0      93     .07       0
Bank Sta=62,93
XS Rating Curve= 0 ,0
Exp/Cntr=0.3,0.1

Type RM Length L Ch R = 1 ,42260.5 ,234.4,263.3,303.7
XS GIS Cut Line= 4
     1567312.184      335048.559      1567345.17      335086.753
     1567451.073      335173.559     1567530.934      335335.017
#Sta/Elev= 30
       0  795.68     8.4  792.62    16.8  789.37    25.2  785.66    42.1  776.25
    50.5  771.99    60.2  768.16      70  765.65    79.8  764.54    89.6  764.46
    99.4  765.06     107   766.2   118.9  768.38   128.7   769.8   138.5  770.95
   148.3  771.89   158.1  772.65   167.8  773.31   187.4  774.37   196.9  774.68
   215.8  775.03   225.3  775.08   282.2   774.8   310.6  775.03   320.1  775.26
   329.6  775.92   339.1  777.58   348.6   780.3     358   783.3   367.5  785.37
#Mann= 3 , 0 , 0
       0     .08       0      70    .045       0     107     .07       0
Bank Sta=70,107
XS Rating Curve= 0 ,0
Exp/Cntr=0.3,0.1

Type RM Length L Ch R = 1 ,41997.2 ,271,266.9,250.6
XS GIS Cut Line= 4
     1567173.295      335206.545     1567204.545      335255.156
     1567218.434      335407.934     1567275.726      335508.628
#Sta/Elev= 25
       0  790.65     9.6  787.52    19.3  783.56    28.9  779.24    38.5  775.04
    48.2  771.78    57.8  770.05    67.4  769.13      77  767.84    86.6  765.96
    96.1  764.57   105.7  764.77     110 765.218   124.9  766.68   134.5  767.29
   144.1  767.73   153.7   768.1   201.6  769.56   230.5  770.63   278.8   772.2
   288.4  772.57   298.1  773.32   307.7  775.53   317.4   779.3     327  783.42
#Mann= 3 , 0 , 0
       0     .08       0    86.6    .045       0     110     .08       0
Bank Sta=86.6,110
XS Rating Curve= 0 ,0
Exp/Cntr=0.3,0.1

Type RM Length L Ch R = 1 ,41730.3 ,170.4,159.6,151.6
XS GIS Cut Line= 3
     1566966.698      335269.045     1566982.323       335347.17
     1567114.267       335597.17
#Sta/Elev= 25
       0  794.42     8.8  792.04    26.6  786.95    35.4  784.36    53.1  778.95
      62  776.03    79.7  769.22    89.4  766.61    99.2  766.01   108.9  765.86
   128.4  765.12   147.9  764.54   177.2  763.43     210 762.334   225.9  762.01
   235.6     762   245.4  762.46     254 763.152   264.9  764.19   274.9  765.24
   303.9  767.88   323.4  769.54   342.9  771.08   352.6  773.36   362.4  777.36
#Mann= 3 , 0 , 0
       0     .06       0     210    .045       0     254     .06       0
Bank Sta=210,254
XS Rating Curve= 0 ,0
Exp/Cntr=0.3,0.1

Type RM Length L Ch R = 1 ,41570.7 ,244.7,240,223.2
XS GIS Cut Line= 3
     1566800.031      335421.823     1566874.684      335465.225
     1567011.837      335694.392
#Sta/Elev= 30
       0  791.02     9.6  787.68    28.8  783.03    38.4  781.31    57.6  777.44
    67.2  775.43    76.8  773.13    86.4  769.71    95.9  766.84   105.4  764.83
     115  765.38     134  767.63   143.6  768.11   153.1  768.22   181.7  767.84
   219.9  766.73   229.4  766.26     237 765.389   248.5  763.64     258   762.8
     266 763.817   267.6  764.02   277.1  766.46   286.7  767.86   305.7  769.44
   315.3  770.67   324.8  773.85   334.4  779.81   343.9  786.39   353.4   792.2
#Mann= 3 , 0 , 0
       0     .08       0     237    .045       0     266     .06       0
Bank Sta=237,266
XS Rating Curve= 0 ,0
Exp/Cntr=0.3,0.1

Type RM Length L Ch R = 1 ,41330.7 ,83.6,106.2,132.8
XS GIS Cut Line= 5
     1566692.392      335529.462     1566718.434      335586.753
     1566900.726      335819.392     1567079.545      335838.489
      1567316.51      336215.819
#Sta/Elev= 30
       0   785.8      45  774.85    91.5   762.1      96 761.617   101.1  761.07
   110.6  760.94     135 761.548   291.8  769.29   339.4  768.63     349  768.69
   358.5  769.69     368  772.36   396.4  782.42   415.3  791.04   434.2  801.31
   443.7  805.75   453.1  808.74   519.4  822.21   538.3  827.85   577.1  833.22
   606.1  835.82   615.8  836.21   644.9  834.93   673.9  834.92   741.7  830.86
   809.5   824.9   848.3  818.97   877.3  815.86   935.5  812.64   983.9  811.03
#Mann= 3 , 0 , 0
       0      .1       0      96    .045       0     135     .06       0
Bank Sta=96,135
XS Rating Curve= 0 ,0
Exp/Cntr=0.3,0.1

Type RM Length L Ch R = 1 ,41224.5 ,41169.1,442.4,438.9
XS GIS Cut Line= 4
      1566626.42      335567.656     1566643.781      335619.739
     1566678.503      335873.212     1566998.584      336338.431
#Sta/Elev= 30
       0  786.87    36.6  773.84      64 762.779    74.6  759.82    84.4  759.23
   104.1   760.5     173  766.97   281.2  767.84   300.9  769.14   330.2  779.18
   349.7  783.56   398.4  803.49   408.1  806.12   417.8  807.33   437.3  807.64
   476.2  806.32   505.5  806.29   524.9  808.88   563.9  817.07   573.6  817.36
   602.8  815.06     632  813.89   661.2   813.3   680.7  813.99   709.9  816.52
   748.9  821.43   778.1  826.07     817  833.52   836.5  835.02   875.4   835.9
#Mann= 3 , 0 , 0
       0      .1       0      64    .045       0   104.1     .06       0
Bank Sta=64,104.1
XS Rating Curve= 0 ,0
Exp/Cntr=0.3,0.1

Type RM Length L Ch R = 1 ,40782.2 ,11618.2,219.1,208.3
XS GIS Cut Line= 4
     1566253.156      335822.864     1566263.573       335847.17
     1566284.406      335946.128     1566464.962      336058.975
#Sta/Elev= 26
       0  778.53     8.8  774.69    17.6  770.31    26.4  765.25    35.6  760.77
    44.8   759.3      54  760.88    63.2  763.22    72.4  765.04    81.6  766.13
    90.8  766.85     100  767.42   109.2  767.86   118.4  768.14   137.2  768.49
   166.3  768.87   195.3  769.41   214.7  769.52   243.7  769.53   263.1  769.68
   282.4  769.99   301.8  770.48   311.5  771.23   321.1  773.52   330.8  777.22
   340.5  781.09
#Mann= 3 , 0 , 0
       0      .1       0    26.4    .045       0    72.4     .09       0
Bank Sta=26.4,72.4
XS Rating Curve= 0 ,0
Exp/Cntr=0.3,0.1

Type RM Length L Ch R = 1 ,40563   ,253,330.1,374.9
XS GIS Cut Line= 4
     1566027.028       335880.59     1566055.674      335924.861
     1566098.628      336021.953     1566114.253      336213.359
#Sta/Elev= 30
       0  787.31    17.6  779.96    26.4  776.12    32.8  773.23    35.2  772.14
    43.9  767.65    52.7  762.95      59 760.664    62.4  759.43      72  758.86
    81.7  759.64      90  760.79     101  762.35   110.6   763.6   120.3  764.73
   129.9  765.75   139.6  766.57   149.2  767.24   158.9  767.87   178.1  768.66
   187.7  769.16   206.9  770.53   254.9  773.58   274.1  774.52   283.7   774.9
   302.9  775.44   312.5  775.92   322.1  776.95   341.3  779.76   350.9  781.44
#Mann= 3 , 0 , 0
       0      .1       0      59    .045       0      90     .07       0
Bank Sta=59,90
XS Rating Curve= 0 ,0
Exp/Cntr=0.3,0.1

Type RM Length L Ch R = 1 ,40233   ,266.7,246.2,209.1
XS GIS Cut Line= 3
     1565873.382       335943.09     1565779.632      336138.403
     1565771.819      336198.298
#Sta/Elev= 23
       0   781.4    18.8   774.5    28.3  770.93    47.1  763.57    56.5   760.4
    65.9  758.39    75.4   760.3    84.8  763.16    94.2  764.63   103.6  764.96
     113   765.1   150.7  764.74   169.6  764.75   188.4  764.95   197.8  765.18
   207.2  765.55   216.6     766   225.3  766.57   233.9  767.62   242.5  769.82
   251.2  773.48   268.4  782.67     277  785.78
#Mann= 3 , 0 , 0
       0      .1       0    47.1    .045       0    84.8     .06       0
Bank Sta=47.1,84.8
XS Rating Curve= 0 ,0
Exp/Cntr=0.3,0.1
