HEC-RAS study SNCHOCRK.prj: SNCHOCRK

--- SNCHOCRK.g02 (geometry) --- (continued)

Type RM Length L Ch R = 1 ,24559.9 ,663.5,664.3,664.3
XS GIS Cut Line= 3
     1568694.562      345822.864     1568709.753      345696.996
     1569028.764      345356.284
#Sta/Elev= 30
       0  752.14     9.8  749.46    19.5  745.74    29.3  741.16    48.8  730.39
    58.5   725.5    68.3  722.45    87.8  720.13    97.5  718.74   107.3  717.85
     117  717.45   204.6  714.24   253.2  712.82   282.4  712.55     331  713.36
   340.7  712.86   350.4  710.83   360.2  709.16   369.9  709.39   379.6   712.5
     399  720.38   408.8  723.79   418.5  726.46   428.2  728.58     506  744.26
   515.7  746.03   544.9  750.71   564.4  754.38   583.8  758.72   593.5  761.68
#Mann= 3 , 0 , 0
       0     .06       0   340.7    .045       0   379.6      .1       0
Bank Sta=340.7,379.6
XS Rating Curve= 0 ,0
Exp/Cntr=0.3,0.1

Type RM Length L Ch R = 1 ,23895.7 ,180.8,183,184.8
XS GIS Cut Line= 3
     1569000.552      346265.573     1569115.569      346198.298
     1569421.559      345874.948
#Sta/Elev= 30
       0  743.45     9.5  743.13      19   742.4    28.6  741.17    47.6  739.53
    57.1  738.34    76.1  735.21    85.7  733.34   114.2  726.82   123.7  725.16
   152.6   722.4   162.3  720.02     172  717.26   181.6  716.17   210.7   715.5
   268.7  715.45   297.8  714.21   317.1  712.49   326.8  710.87   336.5  708.81
   346.2  707.58   355.8  707.82   365.5  709.81   404.2  720.46   413.9  723.73
   433.3  731.34     472  743.89     501  753.66   510.7  757.24   578.4  785.86
#Mann= 3 , 0 , 0
       0     .06       0   317.1    .045       0   365.5      .1       0
Bank Sta=317.1,365.5
XS Rating Curve= 0 ,0
Exp/Cntr=0.3,0.1

Type RM Length L Ch R = 1 ,23712.6 ,404.2,458.4,511.5
XS GIS Cut Line= 3
     1569219.736      346330.677     1569493.174       346068.09
     1570317.826       345918.35
#Sta/Elev= 30
       0  729.74    19.4  725.16    29.2  723.59    38.9  720.71    48.6  716.09
    58.3  712.78    97.2  708.56   116.6  708.43     175  711.32   194.4  711.03
   215.3  709.23   233.3  706.57     243   706.7   252.7  709.02   272.2  716.52
   291.6   722.8   379.1  748.39   564.3  790.08   583.8  793.39   710.5  792.02
   768.9  789.95   827.4  786.72   934.6  776.95  1012.6  774.11  1061.3  771.63
  1080.8  769.74  1129.5  761.73  1178.3  754.85  1197.8   750.6  1217.2  745.05
#Mann= 3 , 0 , 0
       0     .06       0   215.3    .045       0   252.7      .1       0
Bank Sta=215.3,252.7
XS Rating Curve= 0 ,0
Exp/Cntr=0.3,0.1

Type RM Length L Ch R = 1 ,23254.2 ,112,113.5,114.8
XS GIS Cut Line= 5
     1569306.542       346380.59      1569430.24      346476.076
     1569549.597      346512.968     1569958.771      346639.331
     1570502.288      346406.632
#Sta/Elev= 30
       0  724.06    39.1  722.75   107.4  715.01   156.3  711.19   185.1     708
   213.9  707.34   271.6  708.34   300.7  706.78   320.1  705.62   329.9  705.65
   339.6   706.6   349.3  708.53   378.5  712.07   407.7  713.74   631.6  715.28
   670.5  717.68   719.1  723.17   825.7  748.06   903.3  767.86     942  782.24
  1019.6  814.26  1029.3  817.65  1048.7  822.76  1087.4  829.11  1126.2   836.7
  1145.6  836.55  1174.7  841.91  1184.4  842.99  1223.1  845.15  1300.7  843.56
#Mann= 3 , 0 , 0
       0     .06       0   300.7    .045       0   349.3     .06       0
Bank Sta=300.7,349.3
XS Rating Curve= 0 ,0
Exp/Cntr=0.3,0.1

Type RM Length L Ch R = 1 ,23140.7 ,322.7,272.6,222.2
XS GIS Cut Line= 4
      1569287.01      346486.927     1569410.708      346582.413
     1569530.066      346619.305     1569972.774      346756.024
#Sta/Elev= 30
       0  743.25    87.9  734.98   107.4  732.84   156.3  726.01   175.5  722.65
   213.9  717.14   223.5  716.39   271.6  715.93   281.2  715.47   290.8  713.48
   300.5  709.58   310.2  705.86   319.8  704.02   329.5  703.55   339.1  703.57
   348.8  704.46   368.1  708.78   377.7  710.88   387.4  712.43     397  713.37
   416.3   714.2   445.3  714.44   503.2  712.59   532.2  712.39   570.8  713.51
   628.7  716.68     648  717.45     677   717.9   725.2   717.8   744.5  719.24
#Mann= 3 , 0 , 0
       0     .08       0   300.5    .045       0   368.1     .06       0
Bank Sta=300.5,368.1
XS Rating Curve= 0 ,0
Exp/Cntr=0.3,0.1

Type RM Length L Ch R = 1 ,22868.1 ,337.1,348.2,347.6
XS GIS Cut Line= 4
     1569632.062      346942.656     1569842.566      346775.555
     1569987.965      346784.236     1570081.281      346740.833
#Sta/Elev= 30
       0  760.79     9.6  757.83    28.8  750.99    67.2  736.28    76.8  731.93
    86.4  726.41      96  719.96  108.95  710.45   115.2  706.38   124.8  704.06
   134.4  704.96   153.6  709.98   163.2   711.3   182.4  713.08   201.6  714.41
   220.8  715.22   268.8  716.15   307.6  715.99   356.2  716.37   385.3  717.19
     395  717.61   404.7  718.37   414.4  719.38   423.8  720.79   442.5  722.73
   451.8  724.77   461.2  727.98   489.3  738.92   498.6   741.6   517.3  745.87
#Mann= 3 , 0 , 0
       0     .08       0  108.95    .045       0   153.6     .06       0
Bank Sta=108.95,153.6
XS Rating Curve= 0 ,0
Exp/Cntr=0.3,0.1

Type RM Length L Ch R = 1 ,22519.9 ,297.8,324.1,361.9
XS GIS Cut Line= 3
     1569864.267      347124.948     1569959.753      347120.607
     1570250.552      346884.062
#Sta/Elev= 30
       0  738.86     9.6  737.73    19.1  736.32    28.7  734.57    38.2  732.31
    47.8  729.58    66.9   723.5    95.6  714.61   105.2  711.29   114.8   707.2
   124.4   703.9     134  702.35   143.6  702.66   162.9  703.89   210.9  705.93
   249.4  707.86     307  712.41   316.6  713.33   326.3  715.39   335.9  718.24
   345.5  720.04   364.7  724.77   374.3  726.38   383.9  726.47   403.2  732.06
   422.4  736.86     432  740.02   451.2  747.54   460.8  751.14   470.4  754.55
#Mann= 3 , 0 , 0
       0     .07       0   114.8    .045       0   162.9     .06       0
Bank Sta=114.8,162.9
XS Rating Curve= 0 ,0
Exp/Cntr=0.3,0.1

Type RM Length L Ch R = 1 ,22195.8 ,332.3,389.3,438.9
XS GIS Cut Line= 3
     1569946.733      347348.472     1570283.104      347372.343
     1570389.441      347433.107
#Sta/Elev= 30
       0  724.01    38.5  716.91    48.2  715.34    67.4  712.75    86.7  710.88
    96.4  710.35   134.9  709.38   144.5  708.92   154.2  707.98   163.8  706.44
   173.4  704.46     182 702.474   192.7  700.25   202.3  699.28     212  699.19
   240.9  699.88   260.1  699.24     269 699.497   279.4  700.31     289  701.29
   298.7  702.63   308.3  705.02   327.6  711.26   337.2  713.67   346.6  714.85
   356.1  716.86   365.5  720.09   393.7  731.46   450.3   754.9   459.7  759.38
#Mann= 3 , 0 , 0
       0     .08       0     182    .045       0     269     .06       0
Bank Sta=182,269
XS Rating Curve= 0 ,0
Exp/Cntr=0.3,0.1

Type RM Length L Ch R = 1 ,21806.5 ,332,324.3,316.4
XS GIS Cut Line= 4
     1569846.906      347517.743       1569905.5       347547.04
     1569994.476      347706.545     1570079.111      347779.245
#Sta/Elev= 30
       0  732.56     9.4  730.36    18.7  727.49    28.1  723.72    37.4  719.58
    46.8  715.78    56.2  712.32    65.5   709.8    75.1  708.71    84.7  708.37
   123.2  707.62   142.4  707.53     152  707.11   161.6  705.53   180.9  700.28
   190.5  699.39   200.1  700.41   209.7  702.41   219.3  704.47   228.9  706.27
   238.5   707.9   257.4   710.5   266.8   713.6     276  719.82   285.3  727.65
   303.9  743.58   313.2  750.32   322.5  755.35   331.8  759.13   359.7  769.92
#Mann= 3 , 0 , 0
       0     .08       0   161.6    .045       0   209.7     .07       0
Bank Sta=161.6,209.7
XS Rating Curve= 0 ,0
Exp/Cntr=0.3,0.1

Type RM Length L Ch R = 1 ,21482.3 ,262.9,257.6,250.7
XS GIS Cut Line= 4
     1569689.571      347659.887     1569689.571      347816.137
     1569820.865      347984.323     1569963.009      347978.897
#Sta/Elev= 30
       0  739.41     9.8  738.14    19.5  736.39    29.3  734.31    48.8  730.02
    78.1  722.76    97.7   718.6   136.7  711.19   156.2  707.13   187.7  702.42
   204.7  699.55   214.4  698.81   224.1  699.61   233.8  701.62   243.5   703.6
   253.2  704.35   272.6  704.26   282.3  704.45     292  704.77   301.7  705.34
   311.4  706.13   340.5  709.16   350.2   711.1   359.9  714.08   369.6  716.84
   426.5  740.77     436  744.08   445.5  746.88   483.4  756.74   511.9  764.96
#Mann= 3 , 0 , 0
       0      .1       0   187.7    .045       0   233.8     .06       0
Bank Sta=187.7,233.8
XS Rating Curve= 0 ,0
Exp/Cntr=0.3,0.1

Type RM Length L Ch R = 1 ,21224.6 ,224.2,221.1,217.9
XS GIS Cut Line= 2
     1569433.495      347910.538     1569762.271      348240.399
#Sta/Elev= 30
       0  742.28    19.4  736.07    29.1  732.79    38.8  728.51    48.5  723.37
    58.2  717.72    67.9  712.34    77.6  708.41    87.3  706.67   116.4  705.76
   155.2  704.28     165  702.76   174.6  700.32   184.4  698.36     194  698.72
   203.8  699.87   213.5  701.35   223.2  702.47   232.9  703.19   291.1  706.46
   339.6   709.4   349.3  709.78     359  711.38   368.7   714.8   407.5  733.52
   417.2  737.22   426.9  740.21   446.3  745.74     456  748.05   465.7  749.94
#Mann= 3 , 0 , 0
       0      .1       0     165    .045       0   213.5     .07       0
Bank Sta=165,213.5
XS Rating Curve= 0 ,0
Exp/Cntr=0.3,0.1

Type RM Length L Ch R = 1 ,21003.5 ,200.7,201.5,203.7
XS GIS Cut Line= 3
     1569274.532      348079.266     1569647.796      348409.127
     1569769.324      348650.013
#Sta/Elev= 30
       0  756.97    39.1  744.75    48.8  741.38    58.6  736.84    68.4  729.86
    87.9  714.21    97.7     708   107.4  705.41   146.5     705   156.3  704.12
     166  701.48   175.8   698.2   185.6  697.54   216.2  700.37   263.7  700.18
     293  701.06   332.1  704.12   390.7   709.8   410.2  710.48     420  711.37
   429.8  713.83   439.5  717.91   459.1  727.29   468.8  730.49   478.6  732.47
   507.8  733.86   584.8  732.82   652.3  735.47   748.7  741.84   767.9  742.09
#Mann= 3 , 0 , 0
       0      .1       0     166    .045       0   216.2     .06       0
Bank Sta=166,216.2
XS Rating Curve= 0 ,0
Exp/Cntr=0.3,0.1

Type RM Length L Ch R = 1 ,20802.1 ,417.4,406.4,391.3
XS GIS Cut Line= 4
     1569166.025      348246.367     1569343.976      348404.787
     1569450.313       348613.12     1569469.845      348775.881
#Sta/Elev= 30
       0  743.22    19.1  734.02    28.6  728.76    38.1   721.7    47.6  713.84
    57.2  706.69    66.7  702.65    76.2  700.62    85.8  699.49     122 697.762
   133.4  697.15     143  696.96   152.5  697.32     165 698.972   200.1  703.74
   219.2  705.48   238.2  706.51   306.5   709.4     365   713.4   384.4  714.48
   413.7  715.23   442.9  715.06   452.7  715.33   472.2   716.7   481.8  717.92
   491.4  719.53     530   727.9   539.6  729.77   607.2  741.95   636.1  747.68
#Mann= 3 , 0 , 0
       0      .1       0     122    .045       0     165     .08       0
Bank Sta=122,165
XS Rating Curve= 0 ,0
Exp/Cntr=0.3,0.1

Type RM Length L Ch R = 1 ,20395.7 ,354.6,337,337.2
XS GIS Cut Line= 3
     1568890.417      348537.166     1569278.872      348771.541
     1569348.317      348856.176
#Sta/Elev= 30
       0  735.89    19.3  728.22      29  723.72    38.6  718.37    48.3  712.56
    57.9  707.49    67.6  703.69    86.9   699.6    96.5  698.34   106.2  697.44
   120.7  696.84   154.4  695.59   164.1  695.75   190.7  698.12   212.4  700.02
   260.6  704.86   279.9  706.04   318.5  705.53   328.2  705.63   366.8  706.62
   405.4  706.92     444  707.73   462.8  708.21   471.9  708.76     481     710
   499.3  713.74   517.6  718.62   526.7  721.64     554  732.21   563.2   735.1
#Mann= 3 , 0 , 0
       0      .1       0   120.7    .045       0   190.7     .08       0
Bank Sta=120.7,190.7
XS Rating Curve= 0 ,0
Exp/Cntr=0.3,0.1

Type RM Length L Ch R = 1 ,20058.6 ,443.9,460.9,461.2
XS GIS Cut Line= 4
     1568716.806      348884.388     1568825.313      348884.388
     1569126.963      349044.978      1569244.15       349075.36
#Sta/Elev= 30
       0  754.07    27.1  739.52    45.2  730.17    54.2  725.68    72.3  717.03
    99.5  704.58   108.5  700.23   118.3  697.01     128  695.84   137.8   696.3
   157.3  698.96   167.1  699.64   215.9  701.81     255  703.16   284.3  703.77
   303.8   703.9   323.3  703.77   333.1  703.56   352.6  702.87   362.4  702.68
   391.7  702.71   401.4  702.94   411.2   703.6   440.5  706.55   450.2   708.3
   459.6  710.92   468.9  714.26   524.7  735.37     562  749.64   571.3  753.05
#Mann= 3 , 0 , 0
       0      .1       0   108.5    .045       0   157.3     .06       0
Bank Sta=108.5,157.3
XS Rating Curve= 0 ,0
Exp/Cntr=0.3,0.1

Type RM Length L Ch R = 1 ,19597.7 ,241.5,241.7,240
XS GIS Cut Line= 2
     1568690.765      349303.225     1569070.539      349502.877
#Sta/Elev= 30
       0  739.64     9.8  734.46    19.5  728.14    29.2  720.77      39  713.57
    48.8  706.64    58.5   700.3    62.7  698.46    68.3  696.01      78  694.43
    87.8   694.4   107.3  694.51     117  696.82   126.8  699.39   136.5   700.5
   146.3  700.47     156  699.96   175.5  699.28   185.3  699.32   204.8  700.03
   243.8  701.72   302.3   704.7     312  705.55   321.8  707.83   331.5   711.9
     351  721.49   370.6  731.29   399.8   746.1   419.3   755.8   429.1  760.34
#Mann= 3 , 0 , 0
       0      .1       0    62.7    .045       0     117     .06       0
Bank Sta=62.7,117
XS Rating Curve= 0 ,0
Exp/Cntr=0.3,0.1

Type RM Length L Ch R = 1 ,19356   ,151.9,153.2,157.8
XS GIS Cut Line= 4
     1568608.299      349377.009      1568619.15      349509.388
     1568873.056      349628.745     1568966.372       349696.02
#Sta/Elev= 30
       0  755.39     9.5  753.56      19   751.2    28.5  748.24      38  744.44
    56.9  735.54    66.4  731.48    94.9  720.28   132.8  706.59   152.2   702.2
   161.8  700.29   171.5  699.04   219.9  697.35   239.2  697.21   258.6  696.67
   279.5  695.58   297.3  694.57     307   694.4   316.6  694.49   326.3  695.67
     336  697.61   345.7   699.2   355.3   700.1     423  705.01   432.6  706.06
   442.1  708.04   451.7  711.62   461.3  716.15   499.7  734.88   528.4  749.13
#Mann= 3 , 0 , 0
       0     .07       0   279.5    .045       0   326.3     .06       0
Bank Sta=279.5,326.3
XS Rating Curve= 0 ,0
Exp/Cntr=0.3,0.1

Type RM Length L Ch R = 1 ,19202.8 ,239.5,239.3,235.8
XS GIS Cut Line= 3
     1568415.157      349656.957     1568532.345      349607.044
      1568935.99      349824.058
#Sta/Elev= 30
       0  757.43    58.8  742.85    78.4  736.43    88.2  732.55   107.8  724.09
   117.6  720.16   127.4  717.21   137.1  715.76   146.9  713.64   156.6  710.45
   166.4  707.63   176.1  706.03   224.9  702.68   332.1  696.01   351.6   695.3
     389  694.57   400.4  694.41   410.2  694.47     426 695.329   458.9  698.95
   468.6  701.45   478.4  705.56   488.2  710.61   507.6  721.62   536.9  738.99
   546.7  744.48   556.4  749.56   566.2  754.13   575.9  758.14   585.7  761.56
#Mann= 3 , 0 , 0
       0     .06       0     389    .045       0     426     .06       0
Bank Sta=389,426
XS Rating Curve= 0 ,0
Exp/Cntr=0.3,0.1

Type RM Length L Ch R = 1 ,18963.5 ,332.2,332.1,332.7
XS GIS Cut Line= 2
     1568395.626      349787.166     1568847.015        350017.2
#Sta/Elev= 30
       0  748.69     9.7  744.63    19.5  740.09    77.9   712.4    87.7  708.44
    97.4  705.63   107.2   704.9   155.9  704.82   165.6  704.14   175.4  701.96
   185.1  699.28   194.9  697.98   204.6  697.26   243.6  696.82   253.3  696.21
     263  695.92   272.8  696.48     302  696.06     341  696.34   350.7  696.13
   360.5  695.62   370.2   694.7   389.7   694.4   399.4  694.49   409.2  696.16
   418.9  700.72   428.7  706.85   448.2  719.44   496.9  752.35   506.6  758.54
#Mann= 3 , 0 , 0
       0     .06       0   360.5    .045       0   409.2      .1       0
Bank Sta=360.5,409.2
XS Rating Curve= 0 ,0
Exp/Cntr=0.3,0.1

Type RM Length L Ch R = 1 ,18631.4 ,297.6,290,282
XS GIS Cut Line= 4
     1568274.098      350110.516     1568371.754      350136.558
     1568656.042      350292.808     1568723.317      350277.617
#Sta/Elev= 30
       0  739.22     9.2  737.71    18.4  735.71    36.8  730.64    45.9  727.66
    55.1  724.21    82.7   712.6    91.9  709.76   101.1  708.28   179.7  701.98
   228.9   698.8   248.5  697.82   268.2  697.07   297.7  696.15   327.2  695.57
     342 695.005   356.6  694.48   366.5  694.75   376.3  695.76     384 696.864
     396  698.82   405.8  701.13   415.6  704.52   425.5  708.81   434.1   714.2
     460  732.38   468.6  737.94   477.2  742.78   485.8  746.73   494.4  749.62
#Mann= 3 , 0 , 0
       0     .06       0     342    .045       0     384      .1       0
Bank Sta=342,384
XS Rating Curve= 0 ,0
Exp/Cntr=0.3,0.1

Type RM Length L Ch R = 1 ,18341.5 ,165.2,165.8,167.3
XS GIS Cut Line= 6
     1568129.241      350402.183       1568228.2      350442.547
      1568321.95      350467.287     1568566.741      350555.829
     1568756.845      350636.558     1568919.606      350699.058
#Sta/Elev= 30
       0  742.41    29.2  731.28    38.9  726.59      68  710.66    77.7  705.72
    87.4  702.76    97.2   701.9   116.6  701.55     136  700.46     165  699.53
   309.9  697.51     358 695.594   377.4  694.47     387  694.61   396.7  695.56
     410 697.778   425.6  699.77   444.9  701.18   513.3  702.69   582.2  703.35
   601.8  704.66   641.2  709.11   680.4  712.22   709.4  713.78   728.8  714.05
   757.8  712.99   796.6  710.61     816  708.02   825.7  707.12     845  707.39
#Mann= 3 , 0 , 0
       0     .06       0     358    .045       0     410      .1       0
Bank Sta=358,410
XS Rating Curve= 0 ,0
Exp/Cntr=0.3,0.1

Type RM Length L Ch R = 1 ,18175.7 ,183.5,191.3,197.4
XS GIS Cut Line= 6
     1568056.325      350545.412     1568155.283      350585.777
     1568249.033      350610.516     1568493.825      350699.058
     1568683.929      350779.787     1568846.689      350842.287
#Sta/Elev= 30
       0  721.37     9.7  714.84    19.4  709.44    29.2  706.01    38.9   704.3
      68  699.91    87.4  699.28   145.7  698.76   184.4  698.83   271.3  699.82
   319.5  699.62   358.1  698.41   415.9  695.55   425.6   694.8   444.9   694.4
   483.8  694.43   493.6  694.86     533  700.61   542.8  702.52   552.7  705.25
   582.2  714.62     592  716.58   611.7   718.7   641.2  720.58   670.7  724.66
   680.4  725.42   709.4  726.27   786.9  731.89   825.7  735.62     845  736.27
#Mann= 3 , 0 , 0
       0     .06       0   415.9    .045       0   493.6      .1       0
Bank Sta=415.9,493.6
XS Rating Curve= 0 ,0
Exp/Cntr=0.3,0.1

Type RM Length L Ch R = 1 ,17984.5 ,358.6,361,363.7
XS GIS Cut Line= 4
     1567976.898      350607.912     1568023.773      350654.787
     1568483.408      350909.995     1568518.564       350988.12
#Sta/Elev= 30
       0  736.91     9.5  732.38    18.9   727.3    28.4  720.11    37.9  713.21
    47.4  709.84    56.8  707.82    66.3  703.15      76  699.59    85.8  698.65
   153.9  697.22   202.6  697.09   270.7  697.27   319.4  698.79   348.6  698.99
   368.1  698.69   387.6  698.15   474.9  694.81   504.4  693.62   514.1  693.61
   523.9  694.12   533.6   695.1   562.8  697.98   572.6  699.17   582.3  701.08
   611.1  709.38   639.6  718.22   649.1  720.38   658.7  721.74   677.7  723.64
#Mann= 3 , 0 , 0
       0     .08       0   474.9    .045       0   533.6      .1       0
Bank Sta=474.9,533.6
XS Rating Curve= 0 ,0
Exp/Cntr=0.3,0.1

Type RM Length L Ch R = 1 ,17623.5 ,309.4,308.3,298.3
XS GIS Cut Line= 3
     1567841.481      350917.808     1568295.908      351199.058
     1568333.668      351264.162
#Sta/Elev= 30
       0  724.01     9.7  718.92    29.2  707.88    38.9  702.58    48.6  698.46
    58.3  696.78      68  696.78    87.4  697.03   106.9  697.13   155.5  698.11
   184.6  698.46   291.5  698.53   320.6  698.77   340.1  698.83   349.8  698.62
   359.5   697.2     364 695.641   369.2  693.84     379  692.14   388.7   691.9
     395 692.049   456.7  693.87   505.3  695.43     515  696.58   524.7  699.84
   543.8  709.56     572  724.31   590.9  733.89   600.3  737.91   609.7  741.28
#Mann= 3 , 0 , 0
       0     .06       0     364    .045       0     395     .09       0
Bank Sta=364,395
XS Rating Curve= 0 ,0
Exp/Cntr=0.3,0.1

Type RM Length L Ch R = 1 ,17315.2 ,329.3,295.9,267.4
XS GIS Cut Line= 6
     1565645.358      350228.405       1567728.2      350812.339
     1567775.075      351098.797     1567756.845      351192.547
       1568165.7      351421.714     1568282.887      351429.527
#Sta/Elev= 30
       0  795.98   167.2  777.32   265.5   753.9   344.1  725.94     413  752.23
   491.6  760.26   678.4  749.78   757.1  720.14   776.8  716.86   924.2  725.63
  1032.4  723.82  1111.1  728.48  1209.4  721.84  1376.6  725.51  1435.5  716.42
  1553.5  728.47  1720.7  731.28  1828.8  723.47  1907.5  731.04  2163.2  732.27
  2240.6  717.81  2366.3   732.5    2463  727.19  2548.9  697.45  2578.2  694.24
  2705.2   698.5  2945.6  695.65  2978.6  691.84  3007.9  695.51  3135.1  767.09
#Mann= 3 , 0 , 0
       0     .06       0  2945.6    .045       0  3007.9     .08       0
Bank Sta=2945.6,3007.9
XS Rating Curve= 0 ,0
Exp/Cntr=0.3,0.1

Type RM Length L Ch R = 1 ,17019.3 ,436.6,398.3,358.2
XS GIS Cut Line= 6
     1565384.941      351124.239     1566802.157      351165.164
     1567597.991      351755.047     1567736.012      351710.777
     1568142.262      351656.089     1568264.137      351582.478
#Sta/Elev= 30
       0  768.87    68.4  770.33   136.9  790.68   234.7  810.29   361.8  818.14
   567.1   807.9   635.6  786.14   723.6  743.32   831.1  782.66   958.2  806.16
  1163.6  804.34  1329.8  785.76  1378.7   792.6  1545.3   798.4  1702.2  783.72
  1878.8  757.34  1908.2  743.47  1947.4  716.08  1967.1  709.87  2025.9  715.38
    2124  734.83  2231.9  740.06  2320.2  736.64    2534  701.79  2817.7 691.631
  2846.2  691.02  2870.7 691.903  2953.5  697.39  3039.2  742.17  3105.7  769.75
#Mann= 3 , 0 , 0
       0     .06       0  2817.7    .045       0  2870.7     .08       0
Bank Sta=2817.7,2870.7
XS Rating Curve= 0 ,0
Exp/Cntr=0.3,0.1

Type RM Length L Ch R = 1 ,16621   ,561.4,546.2,528.8
XS GIS Cut Line= 2
     1567960.318      352216.159     1568366.134      351717.027
#Sta/Elev= 30
       0  740.51    19.5  731.71      39  723.37    58.5  715.94    68.2     713
      78  710.62    87.7  708.79     117     705   126.7  703.06     156  695.73
   165.7  692.84   175.4  690.96   185.2  690.41   194.9   690.4   233.9   690.4
   243.7  690.65   253.4   691.6   263.2  692.96   272.9  693.86   282.7  694.28
   341.1   694.8   409.4  695.89   419.1  696.78   428.9  698.23   497.1  709.92
   506.8  712.18   516.6  715.34     614  755.95   633.5  763.85   643.3  767.44
#Mann= 3 , 0 , 0
       0     .08       0   165.7    .045       0   253.4     .07       0
Bank Sta=165.7,253.4
XS Rating Curve= 0 ,0
Exp/Cntr=0.3,0.1

Type RM Length L Ch R = 1 ,16074.8 ,627.9,672.3,702.7
XS GIS Cut Line= 4
     1568502.852      352417.981     1568541.915      352357.218
     1568652.592      352053.398     1568669.953      351875.447
#Sta/Elev= 30
       0  724.04    27.1  717.52    36.1   715.5    72.2   708.8      82  706.44
   111.4  697.51   121.2  694.12     131  691.07   140.8  690.24   150.6  690.71
   160.4  693.46   170.2  695.99   172.1  696.08     180  696.48   199.6  695.33
   209.4  695.04   268.2   694.4   287.8  694.46   317.2  694.82   366.2     695
     376  695.15   385.8  695.89   395.6   698.4     405  702.18   414.4  706.52
   423.8  711.01   527.3  761.66   536.7  765.96   546.2  769.77   574.4  779.87
#Mann= 3 , 0 , 0
       0     .07       0   111.4    .045       0   172.1     .07       0
Bank Sta=111.4,172.1
XS Rating Curve= 0 ,0
Exp/Cntr=0.3,0.1

Type RM Length L Ch R = 1 ,15402.6 ,264.6,268.2,285.2
XS GIS Cut Line= 4
     1568880.457      352619.804     1569008.495       352543.85
     1569173.425      352485.256     1569260.231        352387.6
#Sta/Elev= 25
       0  706.63    27.9  705.02     121  700.11   168.3  697.42   197.5  695.61
   216.9  694.26   236.4  692.77   264.4  690.46   275.3  689.47     285   688.8
   294.7  689.01   304.4  691.05   314.2  694.94   323.9  699.53   333.2  703.32
   342.6  707.29   351.9  711.63   361.2  716.32   389.2  730.73   398.6  734.96
   407.9  738.63   417.2  741.65   435.9  748.18   445.2  750.28   454.6  751.51
#Mann= 3 , 0 , 0
       0     .06       0   264.4    .045       0   304.4      .1       0
Bank Sta=264.4,304.4
XS Rating Curve= 0 ,0
Exp/Cntr=0.3,0.1

Type RM Length L Ch R = 1 ,15134.4 ,219.9,210.7,193
XS GIS Cut Line= 4
     1568945.561      352765.204     1569108.321      352780.395
     1569342.696      352715.291     1569492.436       352543.85
#Sta/Elev= 30
       0   703.2     9.6  701.93    19.2   701.2    28.8   700.8    38.5  700.54
    76.9   699.8   115.4  698.56   173.2  696.23   276.6  691.59     290  690.69
   309.4  688.95   319.2  688.85   328.9  691.21   338.6  696.73   348.3   702.8
   358.1  707.97   377.5  717.73   387.3  722.55     397  726.77   406.7  729.53
   416.2  731.04     530  743.18   539.5  743.98     549   744.5     568   744.8
   577.4  745.14   586.9  745.86   605.9  747.68   624.9  749.84   634.3  751.04
#Mann= 3 , 0 , 0
       0     .06       0   276.6    .045       0   328.9      .1       0
Bank Sta=276.6,328.9
XS Rating Curve= 0 ,0
Exp/Cntr=0.3,0.1

Type RM Length L Ch R = 1 ,14923.6 ,157.8,165.6,196.4
XS GIS Cut Line= 3
     1569064.918      353058.172     1569327.505      352932.304
     1569972.188      352274.116
#Sta/Elev= 30
       0  734.67    19.4  732.65    29.1  730.07      68  710.96   106.8  696.26
   116.5  694.92   227.6  691.11   262.1   687.4   271.8  688.66   281.5  692.16
   310.8  703.83   340.2  719.01     350  722.44   359.8  723.96   457.8  731.87
   526.4  735.26   575.4  735.97   614.6   733.4   634.2  733.42     693  740.84
     742  744.06   761.7  748.25   820.5   763.6   849.9  767.66   889.1  776.51
   987.1  803.85  1016.5  809.79  1104.7  838.04  1134.1  842.58  1212.5  850.26
#Mann= 3 , 0 , 0
       0     .06       0   227.6    .045       0   281.5      .1       0
Bank Sta=227.6,281.5
XS Rating Curve= 0 ,0
Exp/Cntr=0.3,0.1

Type RM Length L Ch R = 1 ,14758   ,428.6,497.4,551.4
XS GIS Cut Line= 4
     1569101.811      353127.617     1569188.616      353147.148
     1569338.356      353101.575     1570133.647      353323.595
#Sta/Elev= 30
       0  729.64    35.6  714.59    62.3  705.08    80.1  696.71      89   693.4
    98.8  691.99   108.5  691.88   184.2  692.75   196.6  690.54   216.2     685
   225.9  685.24   245.5  689.48   294.6  700.94   304.5  704.15   343.8  721.06
   353.6  723.53   432.3   738.1   520.7  757.81   609.2  787.71   648.5  799.52
   815.6  841.41   864.8  847.67   913.9   849.7   933.6   849.1   982.7  845.04
  1002.4  841.52    1022  836.49  1031.9  835.63  1051.5   836.5  1071.2  838.97
#Mann= 3 , 0 , 0
       0     .06       0   184.2    .045       0   245.5      .1       0
Bank Sta=184.2,245.5
XS Rating Curve= 0 ,0
Exp/Cntr=0.3,0.1

Type RM Length L Ch R = 1 ,14260.6 ,344.3,410,469.6
XS GIS Cut Line= 3
     1569130.023      353218.763     1569162.575      353379.353
     1569340.526      353700.534
#Sta/Elev= 30
       0  716.99    19.3  714.47    38.6   713.4    67.5  710.05    96.4  707.85
   134.9  703.39   154.2  701.42   173.5  698.88   212.2  692.85   221.8  691.92
   241.2  691.25   260.5     691   308.8  691.13   337.8  690.51   357.1  689.68
   366.8  688.77   376.4   687.1   386.1     685   395.8  683.43   405.4  683.38
   415.1  685.46   424.8  688.64   434.4  691.75   453.7  697.46   463.4  700.87
   473.1  706.42   482.7  713.68   492.4  720.06     502  725.36     531  739.04
#Mann= 3 , 0 , 0
       0     .06       0   376.4    .045       0   424.8      .1       0
Bank Sta=376.4,424.8
XS Rating Curve= 0 ,0
Exp/Cntr=0.3,0.1

Type RM Length L Ch R = 1 ,13850.6 ,345.3,357.9,374.5
XS GIS Cut Line= 4
      1569088.79      353223.103     1569071.429      353296.888
     1568897.818      353479.179     1568845.734      353565.876
#Sta/Elev= 30
       0  713.97    28.4  708.84    37.9  706.78    75.8  697.83    85.5  695.37
    95.2  693.82   104.8  693.39   143.6  694.89   162.9  695.04   172.6  694.79
   230.7   691.6   240.4  690.84   250.1  689.74   262.1  687.96   269.4  686.73
   288.8  682.88   298.5  681.95   308.2  682.35   317.8  684.33   332.1  688.06
   336.7  689.34   345.9   692.6   355.1  698.08   364.3  707.08   373.5  716.67
   391.9  735.02   401.1  743.18   410.3  751.89   419.5  758.65   428.7  764.46
#Mann= 3 , 0 , 0
       0     .06       0   262.1    .045       0   332.1      .1       0
Bank Sta=262.1,332.1
XS Rating Curve= 0 ,0
Exp/Cntr=0.3,0.1

Type RM Length L Ch R = 1 ,13492.7 ,593.5,567.9,542.1
XS GIS Cut Line= 4
     1568929.068      352990.356     1568827.505      353095.824
     1568694.693       353180.46     1568637.401       353249.47
#Sta/Elev= 30
       0  730.53     9.8   728.9    29.3  725.35    48.8  721.44    58.6  719.33
    78.1  714.74    87.8  712.28   107.4  707.11   126.9  701.64   136.7  699.04
   146.4  696.94   155.7   695.6   183.5  692.58     202  690.33   211.3  688.89
   220.5  687.08   229.8  684.77   239.1  682.33   248.3  681.03   257.6  681.83
   266.8  684.51   276.1  687.92   303.9  696.49   312.9  699.68   348.8  712.81
   357.7  715.77   366.7  718.32   375.7  720.58   384.6   722.5   393.6  724.24
#Mann= 3 , 0 , 0
       0     .06       0   220.5    .045       0   276.1     .06       0
Bank Sta=220.5,276.1
XS Rating Curve= 0 ,0
Exp/Cntr=0.3,0.1

Type RM Length L Ch R = 1 ,12924.9 ,230.9,188.9,146.8
XS GIS Cut Line= 3
     1568387.401      352698.689     1568287.141      352886.189
     1568272.818       353086.71
#Sta/Elev= 30
       0  749.12     9.7     744    19.3  738.34      29  732.16    38.7  725.41
    48.3  718.24      58  710.81    67.6  702.93    77.3  694.08      87  685.68
    96.6  681.14   106.3  681.34   125.6  684.39   135.3  685.65   164.3  688.84
   193.3  692.47     203  693.44   212.6  694.18   231.8  695.11   241.3  695.34
   260.5  695.33   298.8  694.84   308.4  694.91   317.9  695.78   327.5  697.99
   356.2  706.34   365.8   708.9   375.4  710.58   384.9   711.4   413.6  712.79
#Mann= 3 , 0 , 0
       0     .08       0      87    .045       0   125.6     .06       0
Bank Sta=87,125.6
XS Rating Curve= 0 ,0
Exp/Cntr=0.3,0.1

Type RM Length L Ch R = 1 ,12735.9 ,248.8,221.1,192.9
XS GIS Cut Line= 3
     1568118.448      352665.037     1568233.032      352984.482
     1568239.976      353073.023
#Sta/Elev= 30
       0  760.55     9.7  755.44    19.4  749.43    29.1  742.41    67.9  712.59
    77.6  704.92    87.3  696.45      97  687.63   106.7  681.71   116.4  680.79
   135.8  683.85   144.8  684.97   174.5  688.17   184.2  689.42   203.6  692.18
   213.3  693.25     223  694.03   232.7  694.59   252.1  695.27   261.8  695.38
     320   694.8   329.7  694.96   339.4  695.71   348.2  697.38   357.1  699.84
   374.9  705.08   383.8   707.4   392.7  709.03   401.5  709.95   428.2  711.27
#Mann= 3 , 0 , 0
       0      .1       0      97    .045       0   144.8     .06       0
Bank Sta=97,144.8
XS Rating Curve= 0 ,0
Exp/Cntr=0.3,0.1

Type RM Length L Ch R = 1 ,12514.8 ,446.1,414.8,384
XS GIS Cut Line= 2
     1567912.141       352843.22     1568224.641      353090.616
#Sta/Elev= 30
       0  736.51    19.4  725.02    58.3   702.3      68  696.27    77.8  689.24
    87.5  682.98    97.2  680.46   106.9  681.39   116.7  683.22   126.4  685.26
   155.5  690.39   165.3  691.74     175   692.8   184.7  693.58   194.4  694.11
   204.2  694.48   213.9   694.6   223.6  694.61     243  694.17   252.8  694.15
   262.5  694.36   272.2  695.14   281.9  697.34   291.6  699.98   301.4  702.25
   311.1  703.71   320.8  704.94   340.2  706.98   359.7  708.86   398.6  711.75
#Mann= 3 , 0 , 0
       0      .1       0    77.8    .045       0   126.4     .06       0
Bank Sta=77.8,126.4
XS Rating Curve= 0 ,0
Exp/Cntr=0.3,0.1

Type RM Length L Ch R = 1 ,12099.9 ,110.5,120,120.2
XS GIS Cut Line= 2
     1567788.443      353297.647      1568149.12      353317.179
#Sta/Elev= 30
       0  735.05     9.8  730.03    19.5  724.89      39  714.38    58.6  704.04
    68.3  698.82    78.1  693.21    87.9  687.04    97.6  681.97   107.4  679.79
   117.2  679.73   136.7   680.9   140.8  681.23   156.2  682.57     166  683.21
   185.5  683.92   195.2   684.5     205  685.64   214.8  687.15   224.5  688.48
   234.3  689.57   244.1   690.8   263.6  693.89   273.3  695.12   283.1  695.88
   292.9  696.43   302.6   697.1   322.2  698.62   351.4  700.13   361.2  700.72
#Mann= 3 , 0 , 0
       0      .1       0    87.9    .045       0   140.8     .06       0
Bank Sta=87.9,140.8
XS Rating Curve= 0 ,0
Exp/Cntr=0.3,0.1

Type RM Length L Ch R = 1 ,11979.9 ,224.4,240.6,266
XS GIS Cut Line= 4
     1567828.807      353401.814     1567860.057      353421.345
     1568013.703       353430.46      1568117.87      353491.658
#Sta/Elev= 24
       0  711.85     9.2  708.52    18.4  704.56    36.6  695.86    46.5  690.62
    56.1  684.81    65.7  680.59    75.3  679.55      85  680.84    94.6   683.1
   104.2  685.39   113.8  687.48   123.4  689.45     133  691.09   142.7  692.08
   152.3  692.59   227.9  695.55   237.2  696.05   246.5  697.37   255.8  699.83
   283.7  709.72     293  713.38   302.3  717.44   311.6  721.83
#Mann= 3 , 0 , 0
       0      .1       0    56.1    .045       0    94.6     .06       0
Bank Sta=56.1,94.6
XS Rating Curve= 0 ,0
Exp/Cntr=0.3,0.1

Type RM Length L Ch R = 1 ,11739.3 ,355.9,398.6,440.7
XS GIS Cut Line= 3
     1567740.266      353513.793     1567813.182      353610.147
     1568082.713      353776.814
#Sta/Elev= 30
       0  709.25    27.9  704.53    55.8   700.6    74.4  698.22   102.2  694.48
   130.4  690.37   188.1  681.47   197.7  679.77   207.3  678.52   216.9  678.13
   226.5  678.97   236.1  681.11   245.7   683.6   255.3  685.17   264.9  686.09
   284.1  687.44   293.7  689.28   303.3  693.31   312.9   698.3   322.5  703.82
   341.7  715.55   351.3  721.17   360.9  726.26   370.5  730.85   380.1  735.08
   389.7  739.02   399.3  742.66   408.9  745.97   428.1  751.83   437.7  754.62
#Mann= 3 , 0 , 0
       0      .1       0   188.1    .045       0   236.1     .06       0
Bank Sta=188.1,236.1
XS Rating Curve= 0 ,0
Exp/Cntr=0.3,0.1

Type RM Length L Ch R = 1 ,11340.7 ,408.9,370.7,332.7
XS GIS Cut Line= 3
     1567546.255      353664.835     1567569.693      353763.793
     1567599.641      353935.668
#Sta/Elev= 16
       0  709.62    27.7  704.24    64.7  697.26   101.7  690.73     152   682.5
   169.5  679.44   179.2  678.19   188.9  678.62   198.6  682.23   208.3  689.13
     218  696.64   227.7  703.21   247.1  716.08   256.8  722.16   266.5  726.63
   276.2  728.88
#Mann= 3 , 0 , 0
       0      .1       0     152    .045       0   198.6      .1       0
Bank Sta=152,198.6
XS Rating Curve= 0 ,0
Exp/Cntr=0.3,0.1

Type RM Length L Ch R = 1 ,10970   ,343.5,311.9,279.8
XS GIS Cut Line= 2
     1567125.682       353836.71     1567426.463      354060.668
#Sta/Elev= 22
       0  742.22     9.6  736.04    19.2  729.61    48.1  709.28    67.3  696.62
    76.9  691.05    86.5  686.54    96.2  683.28   105.8     681   115.4  679.31
     125  678.19   134.6  677.74   144.2   678.2   153.8  679.43   163.5  680.78
   192.3  684.56   288.5  697.49   298.1  699.01   326.9  704.48   336.5  706.22
   365.4  711.12     375  712.65
#Mann= 3 , 0 , 0
       0      .1       0   105.8    .045       0   163.5      .1       0
Bank Sta=105.8,163.5
XS Rating Curve= 0 ,0
Exp/Cntr=0.3,0.1

Type RM Length L Ch R = 1 ,10658.1 ,282.5,264.6,246.5
XS GIS Cut Line= 2
     1567089.224      354220.824     1567384.797      354223.429
#Sta/Elev= 16
       0  730.79    38.1  709.55    57.2  699.02    66.7  693.58    85.8  681.58
    95.4  678.13   104.9  677.92   114.4  678.99   132.8  681.73   200.2  690.55
   219.3  692.98   228.8  694.24   238.4  695.62   247.9  697.19   257.4   698.9
   295.6  705.98
#Mann= 3 , 0 , 0
       0      .1       0    85.8    .045       0   132.8      .1       0
Bank Sta=85.8,132.8
XS Rating Curve= 0 ,0
Exp/Cntr=0.3,0.1

Type RM Length L Ch R = 1 ,10393.6 ,201.1,197.4,193.6
XS GIS Cut Line= 2
     1567141.307      354513.793     1567391.307      354422.647
#Sta/Elev= 14
       0  722.01    47.5  698.44      57  693.58    66.5  688.26      76  682.59
    85.5  678.65      95  677.88   104.5  678.72   125.3  681.96   209.1  694.15
   218.6  695.69   228.1  697.61   237.6  699.79   266.1  706.64
#Mann= 3 , 0 , 0
       0      .1       0      76    .045       0   125.3      .1       0
Bank Sta=76,125.3
XS Rating Curve= 0 ,0
Exp/Cntr=0.3,0.1

Type RM Length L Ch R = 1 ,10196.1 ,221.2,211.5,201.4
XS GIS Cut Line= 5
      1566617.87      354877.074      1567124.38      354660.929
     1567219.432      354698.689     1567354.849      354637.491
     1567445.995       354555.46
#Sta/Elev= 30
       0  733.28     9.8  734.57    19.7   734.7    29.5  733.52    49.2  729.91
      59  730.05    88.5   735.9   108.2   738.1   137.7  736.74   157.3  737.38
   304.8  745.66   383.5  751.94   422.9   754.1   442.5  754.84   511.4  754.38
   521.2  753.08     531  750.69   550.7  744.19   625.1  702.42     653  687.41
   662.3  683.33   671.6  680.36   678.9  679.15   708.7  677.16   727.3  677.93
   748.9   680.5   829.9  688.58   867.6  692.95   886.5  697.28   924.2     708
#Mann= 3 , 0 , 0
       0      .1       0   678.9    .045       0   748.9     .09       0
Bank Sta=678.9,748.9
XS Rating Curve= 0 ,0
Exp/Cntr=0.3,0.1

Type RM Length L Ch R = 1 ,9984.6  ,394.7,394.8,395.3
XS GIS Cut Line= 4
     1566762.835      355210.842     1567276.724      354921.345
     1567471.168      354789.401     1567582.279      354732.109
#Sta/Elev= 30
       0  769.98    29.5  761.78    39.3  759.66    88.5  752.32   157.3  738.88
     177  736.55   206.4   734.4   275.2  724.92   314.6  720.12   344.1  717.68
   412.9   714.6     462  713.47   501.4  713.54   550.5   711.1   560.3  710.04
   570.2  710.19     580  708.34   589.8  703.21   609.4  687.02   619.2  682.35
     629  680.66   658.4  677.23   677.9  675.68   687.7  675.64   707.3  676.79
   824.8   686.6   834.4  687.64     844  689.85   872.9  703.04   949.8  740.46
#Mann= 3 , 0 , 0
       0      .1       0   658.4    .045       0   707.3     .08       0
Bank Sta=658.4,707.3
XS Rating Curve= 0 ,0
Exp/Cntr=0.3,0.1

Type RM Length L Ch R = 1 ,9589.8  ,269.6,262.9,249.8
XS GIS Cut Line= 4
     1567276.724      355369.262     1567356.585      355332.804
     1567587.488      355171.345     1567700.335      355169.609
#Sta/Elev= 30
       0  723.03     9.8  719.84    19.5  715.91    29.3  711.58    58.5  697.82
      78  688.75    87.8  684.48    97.5  681.22   107.2  679.34   116.9  678.68
   165.5  676.86     231  674.03     253     673   262.7  672.78   272.4  672.88
   282.1  673.51     301  675.16     321  676.69   340.4  677.96   350.1  678.83
   359.8  680.96   369.5   685.2     379  691.76   397.8  705.06   407.2  711.56
     426  724.29   444.8  736.64   463.6  748.59     473     754   482.4  757.98
#Mann= 3 , 0 , 0
       0     .09       0     231    .045       0     301     .09       0
Bank Sta=231,301
XS Rating Curve= 0 ,0
Exp/Cntr=0.3,0.1

Type RM Length L Ch R = 1 ,9326.9  ,573.7,522.8,477.6
XS GIS Cut Line= 4
     1567492.002      355697.387     1567542.349       355530.72
     1567632.627      355447.387     1567698.599      355344.956
#Sta/Elev= 27
       0  719.03     9.7  716.97      58  707.06    96.7  699.41   135.4  691.95
   164.4  686.56   202.5  679.65   211.9  678.04   224.9  675.98   240.3   673.6
   249.7  672.53   259.2  672.14   268.6  674.29   278.1  678.62   287.5  684.21
     297  689.33   306.3  693.36   315.7  696.78   325.1  699.08   334.4   700.5
   353.2  702.31   362.6   703.5   381.3  706.38   390.7  707.75   400.1  709.47
   409.4   711.7   418.8   714.6
#Mann= 3 , 0 , 0
       0     .07       0   224.9    .045       0   278.1     .08       0
Bank Sta=224.9,278.1
XS Rating Curve= 0 ,0
Exp/Cntr=0.3,0.1

Type RM Length L Ch R = 1 ,8804    ,506.9,488,473.9
XS GIS Cut Line= 2
     1568052.766      355726.901     1567978.113      355353.637
#Sta/Elev= 21
       0  724.88     9.8  720.34    29.3  710.77      39   705.9    78.1  685.66
    87.8  679.93    97.6  674.83   107.4  672.51   117.1  672.57   126.9  674.03
   136.6  675.95   146.4  677.74   156.2  679.25   165.9  680.48     205  685.12
   234.2  688.45   341.6  701.44   351.4  702.94   361.1  704.94   370.9  707.16
   380.7  709.48
#Mann= 3 , 0 , 0
       0     .09       0    87.8    .045       0   136.6     .06       0
Bank Sta=87.8,136.6
XS Rating Curve= 0 ,0
Exp/Cntr=0.3,0.1

Type RM Length L Ch R = 1 ,8316    ,399.2,406.1,408
XS GIS Cut Line= 4
     1568537.141       355530.72     1568498.946      355476.901
     1568427.766      355338.012     1568351.377      355213.012
#Sta/Elev= 23
       0  722.01     9.4  716.97    18.9  711.19    28.3  704.96    37.7  698.49
    47.1   692.2    56.6  685.66      66  679.07    75.8  673.99    85.5  672.38
    95.3  673.63     105  676.18   114.8  678.29   124.5  679.32   134.3  679.85
     183  682.05   192.8  682.41   290.4  686.83     310  687.73   319.7  688.32
   329.5   689.7   339.3     692   368.6  700.46
#Mann= 3 , 0 , 0
       0     .08       0      66    .045       0   114.8     .06       0
Bank Sta=66,114.8
XS Rating Curve= 0 ,0
Exp/Cntr=0.3,0.1

Type RM Length L Ch R = 1 ,7910    ,257.2,311.2,365.6
XS GIS Cut Line= 4
     1568854.849      355469.956     1568877.418      355332.804
     1568762.835      355086.276     1568780.196      354961.276
#Sta/Elev= 30
       0  717.47    37.1  709.48   101.9  692.87   120.5  688.46   148.7  682.57
   177.8  677.29   197.2  673.36     207  671.66   216.7  671.01   226.4  671.26
   236.1   672.1   245.8  673.85   255.5  674.96   294.3  673.81     304  673.86
   333.2  675.21   342.9  676.48   362.3  680.84     372  682.54   391.4  685.22
   401.1  687.15   410.8  689.67   430.3  697.52   469.1  715.68   478.8  719.06
   488.5  721.17   498.2  722.16   507.9  722.04   517.6  720.71     537  716.82
#Mann= 3 , 0 , 0
       0     .09       0   197.2    .045       0   236.1     .08       0
Bank Sta=197.2,236.1
XS Rating Curve= 0 ,0
Exp/Cntr=0.3,0.1

Type RM Length L Ch R = 1 ,7598.8  ,270.9,290.1,296.9
XS GIS Cut Line= 4
     1568952.071       355490.79     1569049.293      355322.387
     1569165.613      355162.665     1569268.043      355063.706
#Sta/Elev= 30
       0  711.73   126.4  688.92   136.1  687.25   145.8  685.91   155.6  684.97
   165.3  684.28   279.1  676.78     298  675.09   312.6  673.53   335.6  670.83
     345  670.38   354.4  670.83   363.8   672.4   373.2  675.29   382.6  678.82
     392  683.99   401.5  690.19   420.5     704     430  711.48   439.5   719.5
     449  728.37   458.5  737.82     468  747.66   477.5  757.82     487  767.76
   496.5  776.93     506  785.07   515.5  791.98     525  797.42   534.5  801.59
#Mann= 3 , 0 , 0
       0     .06       0   312.6    .045       0   373.2     .09       0
Bank Sta=312.6,373.2
XS Rating Curve= 0 ,0
Exp/Cntr=0.3,0.1

Type RM Length L Ch R = 1 ,7308.7  ,200,210.2,231.4
XS GIS Cut Line= 4
     1569007.627      355542.873     1569203.807      355494.262
     1569323.599      355417.873     1569365.266      355370.998
#Sta/Elev= 29
       0   716.1     9.6  714.64    28.9  711.16    38.5   709.3    48.1   707.2
    57.8  704.34    67.4  700.56    86.6   692.4    96.2  689.12   105.9  687.44
   115.5  686.69   125.1  686.13   192.5   682.4   230.5  680.42   249.5   679.3
   258.9  678.64   268.4  677.68   277.9  676.33   291.6  674.23   306.3  671.91
   315.8   670.7   325.2  670.25   334.7  672.07   344.2  676.38   353.2  680.75
   362.1   684.8     389  695.84     398  700.52   406.9  707.18
#Mann= 3 , 0 , 0
       0     .06       0   291.6    .045       0   344.2      .1       0
Bank Sta=291.6,344.2
XS Rating Curve= 0 ,0
Exp/Cntr=0.3,0.1

Type RM Length L Ch R = 1 ,7098.5  ,306.9,346.7,386.2
XS GIS Cut Line= 5
     1569035.404      355683.498     1569139.571      355695.651
     1569252.418      355673.081     1569450.335      355598.429
     1569561.446      355386.623
#Sta/Elev= 30
       0  716.91    47.7  707.97    57.2  705.38    66.7  701.96    95.3  689.97
   104.9  687.15   114.5  685.77   181.6  682.63   296.9  678.57   306.5  677.68
   331.2  673.68   354.6  669.64   364.2  669.15   373.8  670.49   383.4  674.97
   421.9   696.7   431.5   701.7     441  705.89   469.8  712.93   479.3  714.56
   498.4  716.55   555.9  719.82   584.6  720.66   594.1  720.63   603.7  719.72
   632.4  715.98     642  716.12   651.5  717.26   661.1  719.92   670.7  724.01
#Mann= 3 , 0 , 0
       0     .06       0   331.2    .045       0   383.4      .1       0
Bank Sta=331.2,383.4
XS Rating Curve= 0 ,0
Exp/Cntr=0.3,0.1

Type RM Length L Ch R = 1 ,6751.7  ,323.3,333.7,352.4
XS GIS Cut Line= 4
     1569085.752      355858.845     1569170.821      355876.206
     1569481.585      356018.567     1569830.543      356008.151
#Sta/Elev= 30
       0  707.14     9.6  705.09    19.3  702.02    28.9  698.24    57.9  685.61
    67.5  683.16    77.2   682.5   106.4  681.57   233.3   678.2   243.1  677.35
   248.1   676.3   252.8  675.32   272.4  669.54   282.2  668.73   291.9  670.84
   301.7  677.02   311.4  683.47   340.8  699.94   418.9  744.54   428.6  748.98
   438.3  751.61   583.8  771.41   593.5  772.09   622.6  771.72   651.7  772.42
   700.2  774.61   719.6  775.98   729.3  777.01     739  778.72   777.8  788.24
#Mann= 3 , 0 , 0
       0     .06       0   248.1    .045       0   301.7      .1       0
Bank Sta=248.1,301.7
XS Rating Curve= 0 ,0
Exp/Cntr=0.3,0.1

Type RM Length L Ch R = 1 ,6418    ,427.4,461.1,489.8
XS GIS Cut Line= 4
     1569056.238      356134.887     1569071.863      356159.192
     1569238.529       356280.72     1569327.071       356428.29
#Sta/Elev= 29
       0  696.23     9.6  693.89    19.3  688.68    28.9  682.15    38.7  677.33
    48.5  675.48    58.4   675.4      78  675.68   107.5  675.84   136.9  676.33
   146.8  676.36   156.6  675.76   166.4  674.31   168.1  673.95   176.2  672.23
     186  669.97   195.9  668.48   205.7  668.67   215.5  671.01   225.3  675.71
   235.2  680.67   254.3  687.95   273.4  695.59   302.1  707.22   321.2   715.2
   349.9   727.6   388.1  744.59   397.7  747.78   407.3  749.82
#Mann= 3 , 0 , 0
       0     .06       0   168.1    .045       0   225.3      .1       0
Bank Sta=168.1,225.3
XS Rating Curve= 0 ,0
Exp/Cntr=0.3,0.1

Type RM Length L Ch R = 1 ,5956.9  ,294.7,332.7,366
XS GIS Cut Line= 4
     1568745.474      356150.512     1568787.141      356233.845
     1568877.418      356560.234     1568967.544      357156.234
#Sta/Elev= 30
       0  697.72    74.5  686.98    83.8  684.81   112.5  676.01   122.2  674.89
   364.1   677.1   379.9  676.27   383.4  675.85   402.8  669.73   412.5     668
   422.1  669.16   431.8  673.54   499.9  711.93   509.6  715.87   519.3  717.92
     529  718.15   645.7   713.8   694.3  710.12   723.5  705.39   742.9  700.64
   791.5  686.42   801.3  685.62     811  687.14   859.6  704.67   869.3   707.2
     879  708.36   917.9  709.54   966.5  713.64  1005.4  714.22  1034.6  716.35
#Mann= 3 , 0 , 0
       0     .06       0   379.9    .045       0   431.8      .1       0
Bank Sta=379.9,431.8
XS Rating Curve= 0 ,0
Exp/Cntr=0.3,0.1

Type RM Length L Ch R = 1 ,5624.2  ,543,491.8,445
XS GIS Cut Line= 4
     1568689.918      356134.887     1568707.279      356237.317
     1568530.196      356586.276     1568774.836      357177.067
#Sta/Elev= 30
       0   702.4    94.4  687.35   123.5  676.71   133.2  675.11   240.8  674.84
   358.2  675.83   368.4  675.02   397.4  666.54   407.2  666.73     417  670.83
   426.7  677.65   446.3  689.79   465.9  700.37   475.6   704.7   485.4  706.83
   514.9     708   564.1     713   613.3  715.43   682.1   718.1   790.3  718.35
   849.4  719.34   928.1  715.59   957.6   712.9   977.2  712.55  1006.8  707.26
  1016.6  706.34  1036.3  708.61  1085.5   710.1  1105.1  710.22  1134.6  708.63
#Mann= 3 , 0 , 0
       0     .06       0   368.4    .045       0   426.7     .08       0
Bank Sta=368.4,426.7
XS Rating Curve= 0 ,0
Exp/Cntr=0.3,0.1

Type RM Length L Ch R = 1 ,5132.4  ,454.7,435.4,409.7
XS GIS Cut Line= 4
     1568057.974      356299.817     1568104.849      356341.484
     1568240.266      356620.998     1568337.488      356711.276
#Sta/Elev= 30
       0  706.13    17.9   698.4    35.8  691.04    62.7  680.18    72.4  675.63
    82.1   670.6    91.8  666.35   101.5  665.21   111.2  665.78   134.4  669.44
   140.4  670.35   150.1  671.61   159.8  672.57   179.2  674.28   188.9  674.96
   198.6   675.5   227.7  676.85   247.1  677.56   295.7   678.8   324.8  679.66
   353.9  680.88   363.6  681.48   373.3  682.84   401.7  689.23   439.6  696.98
   468.1   702.6   477.6  704.09     487  704.91   496.5  705.08     506   705.1
#Mann= 3 , 0 , 0
       0      .1       0    82.1    .045       0   134.4     .06       0
Bank Sta=82.1,134.4
XS Rating Curve= 0 ,0
Exp/Cntr=0.3,0.1

Type RM Length L Ch R = 1 ,4697    ,293.4,286.7,279.4
XS GIS Cut Line= 3
     1567783.668      356648.776     1568047.557      356839.748
     1568117.002      356931.762
#Sta/Elev= 29
       0  704.86     9.6  701.45    19.2  698.16    38.3  691.75    57.5  685.59
    67.1   682.6    95.8  673.38     115  666.57   124.6  664.39   134.1  664.08
   143.7  665.43   162.9   670.5   164.5  670.83   172.4  672.48     182  673.57
   220.4  674.33   258.7  675.82     297  677.71   306.6  678.69   316.2   681.1
   325.7  684.66     345  692.32   354.6  695.98   364.2  699.34   373.8  702.41
     393  707.88   412.2  712.93   431.4  717.82     441  720.41
#Mann= 3 , 0 , 0
       0      .1       0    95.8    .045       0   164.5     .06       0
Bank Sta=95.8,164.5
XS Rating Curve= 0 ,0
Exp/Cntr=0.3,0.1
